--- U100-00-00.prj (project) ---

Proj Title=U100-00-00
Current Plan=p02
Default Exp/Contr=0.3,0.1
English Units
Geom File=g01
Flow File=f01
Flow File=f02
Flow File=f03
Plan File=p01
Plan File=p02
Plan File=p03
Y Axis Title=Elevation
X Axis Title(PF)=Main Channel Distance
X Axis Title(XS)=Station
BEGIN DESCRIPTION:
Langham Creek (U100-00-00)
(Flood Hazard & Floodway) Model
10-, 2-, 1-, and 0.2% Events
FILENAME: U100_00_00.prj
PREPARED BY:  LAN                                 DATE: 03/13/2014
REVIEWED BY: LJA                                   DATE: 03/14/2014
This model is not yet approved by FEMA however it will be approved and become effective shortly.
Therefore any LOMR/CLOMR must duplicate their project using this model and submit along with the effective
model when submitting for LOMR/CLOMR review.
Please contact HCFCD if you have any questions.  Brian Edmondson: Brian.Edmondson@hcfcd.org or phone at 713-684-4110
STATUS: Final
ADDICKS WATERSHED MODEL UPDATE
HARRIS COUNTY, TEXAS
END DESCRIPTION:
DSS Export Rating Curves= 0
DSS Export Rating Curve Sorted= 0
DSS Export Volume Flow Curves= 0
DXF Filename=.\Models\Hydraulics\3 - Third Submittal\Restudy-Hydraulics-Duplicate Effective\U100-00-00\U100_00_00.
DXF OffsetX= 0
DXF OffsetY= 0
DXF ScaleX= 1
DXF ScaleY= 10

--- U100-00-00.p02 (plan) ---

Plan Title=Effective Floodway 2019
Program Version=4.10
Short Identifier=Eff+FW
Geom File=g01
Flow File=f02
Subcritical Flow
K Sum by GR= 0
Std Step Tol= 0.01
Critical Tol= 0.01
Num of Std Step Trials= 20
Max Error Tol= 0.3
Flow Tol Ratio= 0.001
Split Flow NTrial= 30
Split Flow Tol= 0.02
Split Flow Ratio= 0.02
Log Output Level= 0
Friction Slope Method= 1
Unsteady Friction Slope Method= 2
Unsteady Bridges Friction Slope Method= 1
Parabolic Critical Depth
Global Vel Dist= 0 , 0 , 0
Global Log Level= 0
CheckData=True
Encroach Param=-1 ,0,0, 2
Encroach River=U100-00-00
Encroach Reach=U100-00-00_0383
Encroach Node=113057.3
       1 1501.18 2576.04
Encroach Node=112699
       1 1828.68 2776.44
Encroach Node=112661.3
       1 1857.29 2838.25
Encroach Node=112573.5
       1 1903.95 2644.83
Encroach Node=112538
       1 1937.21 2641.49
Encroach Node=112398.5
       1 1932.01 2581.05
Encroach Node=112249.7
       1 1933.87 2544.78
Encroach Node=112227.7
       1 1933.49 2547.59
Encroach Node=111785
       1 1965.41 2603.97
Encroach Node=110796.4
       1 1906.27 2629.77
Encroach Node=109730.1
       1 1900.34  2704.6
Encroach Node=108775.4
       1 1896.46 2713.69
Encroach Node=107760.3
       1 2611.03  3580.2
Encroach Node=106699.1
       1 2557.39 3722.79
Encroach Node=105654.6
       1 2624.95  3842.5
Encroach Node=104580.3
       1 2628.97    3960
Encroach Node=103683.9
       1 2627.38 3944.25
Encroach Node=103157.1
       1 2633.53 3970.68
Encroach Node=102624.4
       1 2640.66 4174.01
Encroach Node=102304.1
       1 2634.55 4397.38
Encroach Node=102197.2
       1 2622.84 4479.08
Encroach Node=102116.5
       1 2614.32 4542.43
Encroach Node=101930.3
       1    2974 4885.64
Encroach Node=101878.4
       1 2951.77 4851.17
Encroach Node=101828.7
       1 2930.84 4818.31
Encroach Node=101777.7
       1 2908.97 4788.12
Encroach Node=101652.2
       1 2853.93 4701.09
Encroach Node=101602.5
       1 2832.46 4687.68
Encroach Node=101552.3
       1 2812.46 4947.38
Encroach Node=101503.3
       1 2792.23 4622.67
Encroach Node=100582.2
       1 2636.18 4383.41
Encroach Node=99531.3
       1 2767.77 4398.09
Encroach Node=99490.14
       1 2759.49 4350.74
Encroach Node=98634.54
       1 2860.32 3978.61
Encroach Node=97495.54
       1 2860.23 3548.53
Encroach Node=96771.5
       1    2480 3541.78
Encroach Node=96356.5
       1    2680  3795.8
Encroach Node=96331.5
       1    2897 3864.25
Encroach Node=96265.5
       1    3343 3908.57
Encroach Node=96225.5
       1    3451 4385.24
Encroach Node=96004.46
       1 3731.89 4656.49
Encroach Node=95544.38
       1 4073.81 4319.35
Encroach Node=95444.3
       1 4210.12 4436.55
Encroach Node=94911.28
       1 4285.58  4750.5
Encroach Node=94516.37
       1 4669.07 4971.41
Encroach Node=94452.52
       1 4675.21 4977.52
Encroach Node=94396.13
       1 4678.47 4828.64
Encroach Node=94212.15
       1 4681.47 4818.87
Encroach Node=94148.49
       1 4282.62 4602.35
Encroach Node=94049.88
       1 3825.97 4251.96
Encroach Node=93740.3
       1 2676.62 3483.75
Encroach Node=92724.82
       1 3140.18 3593.54
Encroach Node=92213.05
       1 3382.67 3804.64
Encroach Node=91427.11
       1  3640.7 4243.87
Encroach Node=90943.98
       1 3844.63  4352.4
Encroach Node=90469.36
       1 3862.05 4375.68
Encroach Node=89756.23
       1 4152.23  4513.5
Encroach Node=89599.33
       1 4269.71 4624.26
Encroach Node=89511.89
       1 4269.67 4609.54
Encroach Node=89382.33
       1 4252.56  4630.2
Encroach Node=88559.77
       1 4053.69 4878.11
Encroach Node=87976.86
       1 3851.84 4537.38
Encroach Node=87851.38
       1 1826.62 2515.74
Encroach Node=87766.38
       1 1828.81 2517.93
Encroach Node=87061.14
       1 2089.19 2619.07
Encroach Node=86594.29
       1  2226.4 2487.45
Encroach Node=86498.29
       1 2251.55 2412.12
Encroach Node=86345.65
       1 2252.42 2363.45
Encroach Node=86214.69
       1 2241.94 2359.39
Encroach Node=86116.94
       1 2040.18 2408.84
Encroach Node=85584.03
       1 3644.62 4030.49
Encroach Node=84647.29
       1 3775.96 4146.05
Encroach Node=84525.94
       1 3818.53 4146.05
Encroach Node=84358.83
       1 4264.66 4580.75
Encroach Node=83126.72
       1 3864.69  4243.4
Encroach Node=82787.9
       1 4322.48 4702.12
Encroach Node=82691.01
       1 4186.78 4546.77
Encroach Node=82566.91
       1 4163.07 4311.93
Encroach Node=82349.09
       1 4123.48 4321.77
Encroach Node=82288.55
       1 3996.87 4194.28
Encroach Node=82214.41
       1  3989.7 4182.33
Encroach Node=82108.27
       1 4016.65 4192.51
Encroach Node=82016.73
       1 3979.63 4192.26
Encroach Node=81201.59
       1 3694.12 3821.36
Encroach Node=80190.38
       1 3782.77 3932.69
Encroach Node=79381.02
       1 3607.03 3728.99
Encroach Node=78709.89
       1 3052.79 3181.62
Encroach Node=77984.7
       1 1567.58 1697.55
Encroach Node=77900.38
       1 1567.58 1692.74
Encroach Node=77238.62
       1 1144.57 1267.31
Encroach Node=76425.34
       1 1164.82 1292.28
Encroach Node=75591.2
       1 1154.42 1288.07
Encroach Node=75549.38
       1 1454.63 1582.46
Encroach Node=75528.21
       1 1454.63 1582.46
Encroach Node=75445.26
       1  1391.4 1516.39
Encroach Node=75287.42
       1 1151.98 1275.96
Encroach Node=75169.06
       1  954.09 1093.96
Encroach Node=75148.62
       1     955    1100
Encroach Node=75030.15
       1     950    1110
Encroach Node=75026.36
       1     950    1110
Encroach Node=75005.7
       1     950    1095
Encroach Node=74959.69
       1  948.37  1067.2
Encroach Node=74841.23
       1  908.86 1035.42
Encroach Node=74744.11
       1   879.6 1009.01
Encroach Node=74216.28
       1  988.23 1107.69
Encroach Node=73387.53
       1  987.42  1111.9
Encroach Node=73275.78
       1  942.82 1081.05
Encroach Node=73218.35
       1  942.82 1085.99
Encroach Node=73088.5
       1  854.63  983.58
Encroach Node=72791.48
       1  779.91  908.76
Encroach Node=72607.04
       1  754.13  878.97
Encroach Node=72031.7
       1  920.18 1044.62
Encroach Node=71937.8
       1  948.01 1072.82
Encroach Node=71849.88
       1  966.25 1095.24
Encroach Node=71778.68
       1  762.57  924.34
Encroach Node=71758.34
       1  752.72  932.69
Encroach Node=71756.49
       1  752.12  932.22
Encroach Node=71618.56
       1  743.09   907.8
Encroach Node=71580.98
       1 1097.65 1301.54
Encroach Node=71474.76
       1 1142.14  1311.4
Encroach Node=71377.24
       1 1173.11 1357.51
Encroach Node=71022.41
       1 1105.77 1263.83
Encroach Node=70575.73
       1  930.52 1095.12
Encroach Node=70200.7
       1  647.87  810.06
Encroach Node=69460.43
       1   848.8 1032.63
Encroach Node=69001.19
       1  857.08 1031.02
Encroach Node=68180.03
       1  855.18 1020.16
Encroach Node=67130.95
       1  892.37 1115.68
Encroach Node=66957.83
       1  783.67 1008.86
Encroach Node=66850.04
       1  828.42  1038.1
Encroach Node=66665.68
       1  822.63 1022.49
Encroach Node=66117.75
       1  424.61  609.35
Encroach Node=65911.57
       1  633.75  807.97
Encroach Node=65193.2
       1     415  608.72
Encroach Node=64572.4
       1  669.51  853.58
Encroach Node=64058.53
       1  467.31  769.57
Encroach Node=63538.9
       1 1158.14 1347.92
Encroach Node=63161.89
       1 1321.21 1520.62
Encroach Node=62946.27
       1  1862.1 2081.79
Encroach Node=62063.01
       1 1493.35 1707.63
Encroach Node=61771.35
       1 1418.13 1655.99
Encroach Node=61237.47
       1 1372.44  1591.4
Encroach Node=60580.55
       1 1236.15 1490.54
Encroach Node=60029.36
       1 1406.82  1650.9
Encroach Node=59531.67
       1 1560.49 1807.82
Encroach Node=59431.11
       1 1574.44 1804.36
Encroach Node=59303.02
       1  1485.6 1696.56
Encroach Node=59170.38
       1 1138.02 1361.17
Encroach Node=59048.18
       1  1147.9 1361.17
Encroach Node=58916.32
       1 1134.44  1339.3
Encroach Node=58763.71
       1    1077 1295.28
Encroach Node=58379.91
       1 1234.93 1447.17
Encroach Node=58217.4
       1 1229.21 1484.37
Encroach Node=58077.66
       1 1258.98 1450.54
Encroach Node=57389.92
       1  810.55 1090.42
Encroach Node=57319.71
       1  679.14  921.29
Encroach Node=56824.9
       1  658.99  902.25
Encroach Node=56770.67
       1  654.25  892.47
Encroach Node=56407.3
       1  905.76 1209.65
Encroach Node=56080.86
       1  854.21 1087.18
Encroach Node=55795.19
       1  805.07 1033.25
Encroach Node=55639.65
       1  826.87 1059.31
Encroach Node=55604.97
       1  781.41 1011.25
Encroach Node=55455.98
       1   798.1 1017.19
Encroach Node=55208.76
       1  739.87  963.42
Encroach Node=54863.05
       1 1186.36 1402.86
Encroach Node=54591.68
       1 1392.91 1612.86
Encroach Node=54446.93
       1 1245.87 1500.76
Encroach Node=53835.61
       1     697     990
Encroach Node=53287.78
       1  929.19 1170.63
Encroach Node=52978.66
       1 1024.61 1797.64
Encroach Node=52832.13
       1 1099.23    1810
Encroach Node=52321.22
       1 1179.52 1582.71
Encroach Node=51460.62
       1  991.12 1455.46
Encroach Node=51306.21
       1  788.72 1506.45
Encroach Node=51255.05
       1  795.95 1597.02
Encroach Node=51230.64
       1  373.47 1258.74
Encroach Node=50649.96
       1   49.94  1356.5
Encroach Node=50060.86
       1   53.95    1711
Encroach Node=49388.92
       1   49.81 2175.37
Encroach Node=48823.23
       1   79.62 2602.44
Encroach Node=47982.29
       1  926.92 2960.22
Encroach Node=46816.39
       1  661.71  2720.5
Encroach Node=46039.27
       1   284.3 2274.47
Encroach Node=44920.4
       1 1835.06  3396.1
Encroach Node=43528.58
       1 2213.15 4416.23
Encroach Node=42339.98
       1 2378.45 5031.88
Encroach Node=41257.1
       1 3164.27 5837.31
Encroach Node=40140.33
       1 3549.55 6504.76
Encroach Node=39113.75
       1 4139.33 7677.72
Encroach Node=38317.03
       1 4184.55 7660.37
Computation Interval=1HOUR
Output Interval=1HOUR
Run HTab= 0
Run UNet= 0
Run PostProcess= 0
Run WQNet= 0
UNET Theta= 1
UNET Theta Warmup= 1
UNET ZTol= 0.02
UNET ZSATol= 0.05
UNET MxIter= 20
UNET MaxInSteps= 0
UNET DtIC= 0
UNET DtMin= 0
UNET MaxCRTS= 20
UNET WFStab= 2
UNET SFStab= 1
UNET WFX= 1
UNET SFX= 1
UNET DSS MLevel= 4
UNET DZMax Abort= 100
UNET Convert EG Bridges= 0
UNET Use Existing IB Tables=-1
UNET Froude Reduction=False
UNET Froude Limit= 1
UNET Froude Power= 10
UNET Time Slicing=0,0, 5
UNET Junction Losses=0
Instantaneous Interval=1HOUR
DSS File=dss
Write IC File= 0
Write IC File at Sim End=0
Echo Input=False
Echo Parameters=False
Echo Output=False
Write Detailed= 0
WQ AD Non Conservative
WQ ULTIMATE=-1
WQ Max Comp Step=1HOUR
WQ Output Interval=15MIN
WQ Output Selected Increments= 0
WQ Output face flow=0
WQ Output face velocity=0
WQ Output face area=0
WQ Output face dispersion=0
WQ Output cell volume=0
WQ Output cell surface area=0
WQ Output cell continuity=0
WQ Output cumulative cell continuity=0
WQ Output face conc=0
WQ Output face dconc_dx=0
WQ Output face courant=0
WQ Output face peclet=0
WQ Output face adv mass=0
WQ Output face disp mass=0
WQ Output cell mass=0
WQ Output cell source sink temp=0
WQ Output cell source sink nsm=0
WQ Output MaxMinRange=-1
WQ Daily Max Min Mean=-1
WQ Daily Range=0
WQ Daily Time=0
WQ Create Restart=0
WQ Fixed Restart=0
WQ System Summary=0
WQ Use Fixed Temperature=0
Sorting and Armoring Iterations= 10
XS Update Threshold= 0.02
Hydraulics Update Threshold= 0.02
Energy Slope Method= 1
Volume Change Method= 0
XS Weighting Method= 0
Number of US Weighted Cross Sections= 1
Number of DS Weighted Cross Sections= 1
Upstream XS Weight=0.25
Main XS Weight=0.5
Downstream XS Weight=0.25
Number of DS XS's Weighted with US Boundary= 1
Upstream Boundary Weight= 1
Weight of XSs Associated with US Boundary= 0
Number of US XS's Weighted with DS Boundary= 1
Downstream Boundary Weight= 0.5
Weight of XSs Associated with DS Boundary= 0.5
Sediment Output Level= 4
Mass or Volume Output= 0
Output Increment Type= 1
Profile and TS Output Increment= 10
XS Output Flag= 0
XS Output Increment= 10
Disregard all LS=0
Disregard all Conn=0
Disregard all Breaches=0
Disregard all Pumps=0

--- U100-00-00.p01 (plan) ---

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Plan Title=Effective Multi-profile
Short Identifier=Eff+MP
Geom File=g01
Flow File=f01
Encroach Param=-1 ,0,0, 0

--- U100-00-00.p03 (plan) ---

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Plan Title=SVSQ
Short Identifier=SVSQ
Geom File=g01
Flow File=f03
Encroach Param=-1 ,0,0, 0

--- U100-00-00.f02 (steady flow) ---

Flow Title=Effective Floodway 2019
Program Version=4.10
Number of Profiles= 2
Profile Names=100YR,FW
River Rch & RM=U100-00-00,U100-00-00_0383 ,113057.3
     998     998
River Rch & RM=U100-00-00,U100-00-00_0383 ,112249.7
    1022    1022
River Rch & RM=U100-00-00,U100-00-00_0383 ,111785
    1076    1076
River Rch & RM=U100-00-00,U100-00-00_0383 ,110796.4
    1137    1137
River Rch & RM=U100-00-00,U100-00-00_0383 ,109730.1
    1195    1195
River Rch & RM=U100-00-00,U100-00-00_0383 ,108775.4
    1260    1260
River Rch & RM=U100-00-00,U100-00-00_0383 ,107760.3
    1331    1331
River Rch & RM=U100-00-00,U100-00-00_0383 ,106699.1
    1405    1405
River Rch & RM=U100-00-00,U100-00-00_0383 ,105654.6
    1486    1486
River Rch & RM=U100-00-00,U100-00-00_0383 ,104580.3
    1557    1557
River Rch & RM=U100-00-00,U100-00-00_0383 ,103683.9
    1600    1600
River Rch & RM=U100-00-00,U100-00-00_0383 ,103157.1
    1672    1672
River Rch & RM=U100-00-00,U100-00-00_0383 ,102304.1
    1743    1743
River Rch & RM=U100-00-00,U100-00-00_0383 ,101552.3
    1828    1828
River Rch & RM=U100-00-00,U100-00-00_0383 ,100582.2
    1931    1931
River Rch & RM=U100-00-00,U100-00-00_0383 ,99531.3
    1935    1935
River Rch & RM=U100-00-00,U100-00-00_0383 ,99490.14
    1937    1937
River Rch & RM=U100-00-00,U100-00-00_0383 ,97495.54
    2044    2044
River Rch & RM=U100-00-00,U100-00-00_0383 ,95544.38
    2086    2086
River Rch & RM=U100-00-00,U100-00-00_0383 ,93740.3
    2158    2158
River Rch & RM=U100-00-00,U100-00-00_0383 ,91427.11
    2254    2254
River Rch & RM=U100-00-00,U100-00-00_0383 ,89382.33
    2343    2343
River Rch & RM=U100-00-00,U100-00-00_0383 ,87061.14
    2448    2448
River Rch & RM=U100-00-00,U100-00-00_0383 ,85584.03
    2517    2517
River Rch & RM=U100-00-00,U100-00-00_0383 ,84358.83
    2575    2575
River Rch & RM=U100-00-00,U100-00-00_0383 ,82566.91
    2664    2664
River Rch & RM=U100-00-00,U100-00-00_0383 ,82288.55
    2691    2691
River Rch & RM=U100-00-00,U100-00-00_0383 ,81201.59
    2802    2802
River Rch & RM=U100-00-00,U100-00-00_0383 ,79381.02
    2996    2996
River Rch & RM=U100-00-00,U100-00-00_0383 ,77984.7
    3155    3155
River Rch & RM=U100-00-00,U100-00-00_0383 ,76425.34
    3342    3342
River Rch & RM=U100-00-00,U100-00-00_0383 ,74744.11
    3556    3556
River Rch & RM=U100-00-00,U100-00-00_0383 ,73088.5
    3780    3780
River Rch & RM=U100-00-00,U100-00-00_0383 ,71377.24
    4027    4027
River Rch & RM=U100-00-00,U100-00-00_0383 ,71022.41
    6296    6296
River Rch & RM=U100-00-00,U100-00-00_0383 ,70575.73
    6428    6428
River Rch & RM=U100-00-00,U100-00-00_0383 ,69460.43
    6770    6770
River Rch & RM=U100-00-00,U100-00-00_0383 ,69001.19
    6916    6916
River Rch & RM=U100-00-00,U100-00-00_0383 ,68180.03
    7185    7185
River Rch & RM=U100-00-00,U100-00-00_0383 ,67130.95
    7544    7544
River Rch & RM=U100-00-00,U100-00-00_0383 ,65911.57
    7985    7985
River Rch & RM=U100-00-00,U100-00-00_0383 ,65193.2
    8256    8256
River Rch & RM=U100-00-00,U100-00-00_0383 ,64058.53
    8703    8703
River Rch & RM=U100-00-00,U100-00-00_0383 ,63161.89
    8810    8810
River Rch & RM=U100-00-00,U100-00-00_0383 ,58763.71
    9354    9354
River Rch & RM=U100-00-00,U100-00-00_0383 ,54446.93
    9921    9921
River Rch & RM=U100-00-00,U100-00-00_0383 ,50060.86
   10533   10533
River Rch & RM=U100-00-00,U100-00-00_0383 ,49388.92
   19258   19258
River Rch & RM=U100-00-00,U100-00-00_0383 ,48823.23
   19654   19654
River Rch & RM=U100-00-00,U100-00-00_0383 ,43528.58
   20052   20052
Boundary for River Rch & Prof#=U100-00-00,U100-00-00_0383 , 1
Up Type= 0
Dn Type= 1
Dn Known WS=100.8
Boundary for River Rch & Prof#=U100-00-00,U100-00-00_0383 , 2
Up Type= 0
Dn Type= 1
Dn Known WS=101.8
Observed WS=U100-00-00      ,U100-00-00_0383 ,113057.3,0,157.68,157.94
Observed WS=U100-00-00      ,U100-00-00_0383 ,112699  ,0,157.23,157.57
Observed WS=U100-00-00      ,U100-00-00_0383 ,112661.3,0,157.18,157.53
Observed WS=U100-00-00      ,U100-00-00_0383 ,112573.5,0,157.07,157.44
Observed WS=U100-00-00      ,U100-00-00_0383 ,112538  ,0,157.07,157.43
Observed WS=U100-00-00      ,U100-00-00_0383 ,112398.5,0,156.92,157.18
Observed WS=U100-00-00      ,U100-00-00_0383 ,112249.7,0,156.79,156.99
Observed WS=U100-00-00      ,U100-00-00_0383 ,112227.7,0,156.4,156.74
Observed WS=U100-00-00      ,U100-00-00_0383 ,111785  ,0,156.13,156.39
Observed WS=U100-00-00      ,U100-00-00_0383 ,110796.4,0,155.43,155.75
Observed WS=U100-00-00      ,U100-00-00_0383 ,109730.1,0,154.8,154.96
Observed WS=U100-00-00      ,U100-00-00_0383 ,108775.4,0,152.76,153.47
Observed WS=U100-00-00      ,U100-00-00_0383 ,107760.3,0,152.04,152.27
Observed WS=U100-00-00      ,U100-00-00_0383 ,106699.1,0,151.58,151.81
Observed WS=U100-00-00      ,U100-00-00_0383 ,105654.6,0,151,151.27
Observed WS=U100-00-00      ,U100-00-00_0383 ,104580.3,0,150.63,150.9
Observed WS=U100-00-00      ,U100-00-00_0383 ,103683.9,0,150.42,150.69
Observed WS=U100-00-00      ,U100-00-00_0383 ,103157.1,0,150.22,150.47
Observed WS=U100-00-00      ,U100-00-00_0383 ,102624.4,0,150.19,150.44
Observed WS=U100-00-00      ,U100-00-00_0383 ,102304.1,0,150.14,150.38
Observed WS=U100-00-00      ,U100-00-00_0383 ,102197.2,0,149.91,150.29
Observed WS=U100-00-00      ,U100-00-00_0383 ,102116.5,0,149.99,150.29
Observed WS=U100-00-00      ,U100-00-00_0383 ,101930.3,0,149.9,150.23
Observed WS=U100-00-00      ,U100-00-00_0383 ,101878.4,0,149.88,150.21
Observed WS=U100-00-00      ,U100-00-00_0383 ,101828.7,0,149.85,150.2
Observed WS=U100-00-00      ,U100-00-00_0383 ,101777.7,0,149.83,150.18
Observed WS=U100-00-00      ,U100-00-00_0383 ,101652.2,0,149.77,150.14
Observed WS=U100-00-00      ,U100-00-00_0383 ,101602.5,0,149.76,150.14
Observed WS=U100-00-00      ,U100-00-00_0383 ,101552.3,0,149.75,150.13
Observed WS=U100-00-00      ,U100-00-00_0383 ,101503.3,0,149.74,150.13
Observed WS=U100-00-00      ,U100-00-00_0383 ,100582.2,0,149.55,150.04
Observed WS=U100-00-00      ,U100-00-00_0383 ,99531.3 ,0,149.44,149.97
Observed WS=U100-00-00      ,U100-00-00_0383 ,99490.14,0,149.43,149.97
Observed WS=U100-00-00      ,U100-00-00_0383 ,98634.54,0,149.32,149.89
Observed WS=U100-00-00      ,U100-00-00_0383 ,97495.54,0,148.98,149.6
Observed WS=U100-00-00      ,U100-00-00_0383 ,96771.5 ,0,148.26,148.78
Observed WS=U100-00-00      ,U100-00-00_0383 ,96004.46,0,148.09,148.56
Observed WS=U100-00-00      ,U100-00-00_0383 ,95544.38,0,147.71,148.14
Observed WS=U100-00-00      ,U100-00-00_0383 ,94911.28,0,147.08,147.57
Observed WS=U100-00-00      ,U100-00-00_0383 ,94516.37,0,146.64,147.26
Observed WS=U100-00-00      ,U100-00-00_0383 ,94452.52,0,146.56,147.2
Observed WS=U100-00-00      ,U100-00-00_0383 ,94396.13,0,146.5,147.16
Observed WS=U100-00-00      ,U100-00-00_0383 ,94212.15,0,146.31,146.94
Observed WS=U100-00-00      ,U100-00-00_0383 ,94148.49,0,146.24,146.86
Observed WS=U100-00-00      ,U100-00-00_0383 ,94049.88,0,146.14,146.74
Observed WS=U100-00-00      ,U100-00-00_0383 ,93740.3 ,0,145.82,146.37
Observed WS=U100-00-00      ,U100-00-00_0383 ,92724.82,0,144.63,145.04
Observed WS=U100-00-00      ,U100-00-00_0383 ,92213.05,0,143.78,144.08
Observed WS=U100-00-00      ,U100-00-00_0383 ,91427.11,0,142.73,143.17
Observed WS=U100-00-00      ,U100-00-00_0383 ,90943.98,0,142.52,142.96
Observed WS=U100-00-00      ,U100-00-00_0383 ,90469.36,0,142.31,142.75
Observed WS=U100-00-00      ,U100-00-00_0383 ,89756.23,0,142.01,142.44
Observed WS=U100-00-00      ,U100-00-00_0383 ,89599.33,0,141.95,142.37
Observed WS=U100-00-00      ,U100-00-00_0383 ,89511.89,0,141.95,142.33
Observed WS=U100-00-00      ,U100-00-00_0383 ,89382.33,0,141.9,142.27
Observed WS=U100-00-00      ,U100-00-00_0383 ,88559.77,0,141.57,141.92
Observed WS=U100-00-00      ,U100-00-00_0383 ,87976.86,0,140.6,141.06
Observed WS=U100-00-00      ,U100-00-00_0383 ,87851.38,0,140.41,140.95
Observed WS=U100-00-00      ,U100-00-00_0383 ,87766.38,0,140.35,140.9
Observed WS=U100-00-00      ,U100-00-00_0383 ,87061.14,0,139.89,140.49
Observed WS=U100-00-00      ,U100-00-00_0383 ,86116.94,0,139.49,140.1
Observed WS=U100-00-00      ,U100-00-00_0383 ,85584.03,0,138.79,139.56
Observed WS=U100-00-00      ,U100-00-00_0383 ,84647.29,0,137.86,138.99
Observed WS=U100-00-00      ,U100-00-00_0383 ,84525.94,0,137.74,138.92
Observed WS=U100-00-00      ,U100-00-00_0383 ,84358.83,0,137.57,138.82
Observed WS=U100-00-00      ,U100-00-00_0383 ,83126.72,0,134.65,136.81
Observed WS=U100-00-00      ,U100-00-00_0383 ,82787.9 ,0,133.35,135.78
Observed WS=U100-00-00      ,U100-00-00_0383 ,82691.01,0,132.98,135.48
Observed WS=U100-00-00      ,U100-00-00_0383 ,82566.91,0,132.51,135.1
Observed WS=U100-00-00      ,U100-00-00_0383 ,82349.09,0,131.68,134.44
Observed WS=U100-00-00      ,U100-00-00_0383 ,82288.55,0,131.44,134.26
Observed WS=U100-00-00      ,U100-00-00_0383 ,82214.41,0,131.16,134.03
Observed WS=U100-00-00      ,U100-00-00_0383 ,82108.27,0,130.77,133.76
Observed WS=U100-00-00      ,U100-00-00_0383 ,82016.73,0,130.59,132.87
Observed WS=U100-00-00      ,U100-00-00_0383 ,81201.59,0,129.61,131.96
Observed WS=U100-00-00      ,U100-00-00_0383 ,80190.38,0,128.64,131.01
Observed WS=U100-00-00      ,U100-00-00_0383 ,79381.02,0,127.85,130.23
Observed WS=U100-00-00      ,U100-00-00_0383 ,78709.89,0,127.19,129.58
Observed WS=U100-00-00      ,U100-00-00_0383 ,77984.7 ,0,126.47,128.84
Observed WS=U100-00-00      ,U100-00-00_0383 ,77900.38,0,126.39,128.76
Observed WS=U100-00-00      ,U100-00-00_0383 ,77238.62,0,125.76,128.09
Observed WS=U100-00-00      ,U100-00-00_0383 ,76425.34,0,125.04,127.32
Observed WS=U100-00-00      ,U100-00-00_0383 ,75591.2 ,0,124.18,126.43
Observed WS=U100-00-00      ,U100-00-00_0383 ,75549.38,0,124.15,126.39
Observed WS=U100-00-00      ,U100-00-00_0383 ,75528.21,0,123.85,126.12
Observed WS=U100-00-00      ,U100-00-00_0383 ,75445.26,0,123.81,126.07
Observed WS=U100-00-00      ,U100-00-00_0383 ,75287.42,0,123.73,125.98
Observed WS=U100-00-00      ,U100-00-00_0383 ,75169.06,0,123.33,125.45
Observed WS=U100-00-00      ,U100-00-00_0383 ,75148.62,0,123.18,125.26
Observed WS=U100-00-00      ,U100-00-00_0383 ,75030.15,0,123.04,125.05
Observed WS=U100-00-00      ,U100-00-00_0383 ,75026.36,0,122.98,125.05
Observed WS=U100-00-00      ,U100-00-00_0383 ,75005.7 ,0,122.64,125.06
Observed WS=U100-00-00      ,U100-00-00_0383 ,74959.69,0,122.55,124.97
Observed WS=U100-00-00      ,U100-00-00_0383 ,74841.23,0,122.33,124.72
Observed WS=U100-00-00      ,U100-00-00_0383 ,74744.11,0,122.14,124.52
Observed WS=U100-00-00      ,U100-00-00_0383 ,74216.28,0,120.94,123.34
Observed WS=U100-00-00      ,U100-00-00_0383 ,73387.53,0,119.24,121.75
Observed WS=U100-00-00      ,U100-00-00_0383 ,73275.78,0,119.19,121.7
Observed WS=U100-00-00      ,U100-00-00_0383 ,73218.35,0,118.99,121.47
Observed WS=U100-00-00      ,U100-00-00_0383 ,73088.5 ,0,118.78,121.25
Observed WS=U100-00-00      ,U100-00-00_0383 ,72791.48,0,118.31,120.76
Observed WS=U100-00-00      ,U100-00-00_0383 ,72607.04,0,117.78,120.26
Observed WS=U100-00-00      ,U100-00-00_0383 ,72031.7 ,0,117.22,119.82
Observed WS=U100-00-00      ,U100-00-00_0383 ,71937.8 ,0,117.13,119.75
Observed WS=U100-00-00      ,U100-00-00_0383 ,71849.88,0,117.06,119.69
Observed WS=U100-00-00      ,U100-00-00_0383 ,71778.68,0,117.01,119.64
Observed WS=U100-00-00      ,U100-00-00_0383 ,71758.34,0,116.99,119.63
Observed WS=U100-00-00      ,U100-00-00_0383 ,71756.49,0,116.99,119.63
Observed WS=U100-00-00      ,U100-00-00_0383 ,71618.56,0,116.2,118.84
Observed WS=U100-00-00      ,U100-00-00_0383 ,71580.98,0,116.16,118.8
Observed WS=U100-00-00      ,U100-00-00_0383 ,71474.76,0,116.05,118.69
Observed WS=U100-00-00      ,U100-00-00_0383 ,71377.24,0,115.94,118.59
Observed WS=U100-00-00      ,U100-00-00_0383 ,71022.41,0,115.56,118.23
Observed WS=U100-00-00      ,U100-00-00_0383 ,70575.73,0,115.03,117.75
Observed WS=U100-00-00      ,U100-00-00_0383 ,70200.7 ,0,114.58,117.34
Observed WS=U100-00-00      ,U100-00-00_0383 ,69460.43,0,113.97,116.73
Observed WS=U100-00-00      ,U100-00-00_0383 ,69001.19,0,113.66,116.4
Observed WS=U100-00-00      ,U100-00-00_0383 ,68180.03,0,112.96,115.64
Observed WS=U100-00-00      ,U100-00-00_0383 ,67130.95,0,112.36,115.05
Observed WS=U100-00-00      ,U100-00-00_0383 ,66957.83,0,112.21,114.89
Observed WS=U100-00-00      ,U100-00-00_0383 ,66850.04,0,111.93,114.57
Observed WS=U100-00-00      ,U100-00-00_0383 ,66665.68,0,111.75,114.38
Observed WS=U100-00-00      ,U100-00-00_0383 ,66117.75,0,111.21,113.81
Observed WS=U100-00-00      ,U100-00-00_0383 ,65911.57,0,110.89,113.46
Observed WS=U100-00-00      ,U100-00-00_0383 ,65193.2 ,0,110.14,112.7
Observed WS=U100-00-00      ,U100-00-00_0383 ,64572.4 ,0,109.57,112.13
Observed WS=U100-00-00      ,U100-00-00_0383 ,64058.53,0,109.33,112
Observed WS=U100-00-00      ,U100-00-00_0383 ,63538.9 ,0,108.67,111.35
Observed WS=U100-00-00      ,U100-00-00_0383 ,63161.89,0,108.43,111.12
Observed WS=U100-00-00      ,U100-00-00_0383 ,62946.27,0,108.3,110.99
Observed WS=U100-00-00      ,U100-00-00_0383 ,62063.01,0,107.95,110.64
Observed WS=U100-00-00      ,U100-00-00_0383 ,61771.35,0,107.84,110.52
Observed WS=U100-00-00      ,U100-00-00_0383 ,61237.47,0,107.64,110.31
Observed WS=U100-00-00      ,U100-00-00_0383 ,60580.55,0,107.49,110.16
Observed WS=U100-00-00      ,U100-00-00_0383 ,60029.36,0,107.28,109.91
Observed WS=U100-00-00      ,U100-00-00_0383 ,59531.67,0,107.13,109.73
Observed WS=U100-00-00      ,U100-00-00_0383 ,59431.11,0,107.1,109.7
Observed WS=U100-00-00      ,U100-00-00_0383 ,59303.02,0,107.06,109.65
Observed WS=U100-00-00      ,U100-00-00_0383 ,59170.38,0,106.56,108.95
Observed WS=U100-00-00      ,U100-00-00_0383 ,59048.18,0,106.22,108.55
Observed WS=U100-00-00      ,U100-00-00_0383 ,58916.32,0,106.14,108.48
Observed WS=U100-00-00      ,U100-00-00_0383 ,58763.71,0,106.04,108.39
Observed WS=U100-00-00      ,U100-00-00_0383 ,58379.91,0,105.86,108.17
Observed WS=U100-00-00      ,U100-00-00_0383 ,58217.4 ,0,105.78,108.08
Observed WS=U100-00-00      ,U100-00-00_0383 ,58077.66,0,105.59,107.86
Observed WS=U100-00-00      ,U100-00-00_0383 ,57389.92,0,105.2,107.37
Observed WS=U100-00-00      ,U100-00-00_0383 ,57319.71,0,105.2,107.39
Observed WS=U100-00-00      ,U100-00-00_0383 ,56824.9 ,0,104.97,107.13
Observed WS=U100-00-00      ,U100-00-00_0383 ,56770.67,0,104.95,107.11
Observed WS=U100-00-00      ,U100-00-00_0383 ,56407.3 ,0,104.81,106.94
Observed WS=U100-00-00      ,U100-00-00_0383 ,56080.86,0,104.72,106.81
Observed WS=U100-00-00      ,U100-00-00_0383 ,55795.19,0,104.64,106.69
Observed WS=U100-00-00      ,U100-00-00_0383 ,55639.65,0,104.6,106.63
Observed WS=U100-00-00      ,U100-00-00_0383 ,55604.97,0,104.59,106.62
Observed WS=U100-00-00      ,U100-00-00_0383 ,55455.98,0,104.55,106.56
Observed WS=U100-00-00      ,U100-00-00_0383 ,55208.76,0,104.49,106.47
Observed WS=U100-00-00      ,U100-00-00_0383 ,54863.05,0,104.4,106.34
Observed WS=U100-00-00      ,U100-00-00_0383 ,54591.68,0,104.35,106.26
Observed WS=U100-00-00      ,U100-00-00_0383 ,54446.93,0,104.32,106.22
Observed WS=U100-00-00      ,U100-00-00_0383 ,53835.61,0,104.2,106.05
Observed WS=U100-00-00      ,U100-00-00_0383 ,53287.78,0,103.93,105.64
Observed WS=U100-00-00      ,U100-00-00_0383 ,52978.66,0,103.77,105.42
Observed WS=U100-00-00      ,U100-00-00_0383 ,52832.13,0,103.62,105.23
Observed WS=U100-00-00      ,U100-00-00_0383 ,52321.22,0,103.53,105.11
Observed WS=U100-00-00      ,U100-00-00_0383 ,51460.62,0,103.42,104.98
Observed WS=U100-00-00      ,U100-00-00_0383 ,51306.21,0,103.38,104.93
Observed WS=U100-00-00      ,U100-00-00_0383 ,51255.05,0,103.37,104.92
Observed WS=U100-00-00      ,U100-00-00_0383 ,51230.64,0,103.36,104.92
Observed WS=U100-00-00      ,U100-00-00_0383 ,50649.96,0,103.28,104.83
Observed WS=U100-00-00      ,U100-00-00_0383 ,50060.86,0,102.83,104.36
Observed WS=U100-00-00      ,U100-00-00_0383 ,49388.92,0,102.79,104.29
Observed WS=U100-00-00      ,U100-00-00_0383 ,48823.23,0,102.75,104.24
Observed WS=U100-00-00      ,U100-00-00_0383 ,47982.29,0,102.59,104.05
Observed WS=U100-00-00      ,U100-00-00_0383 ,46816.39,0,102.31,103.72
Observed WS=U100-00-00      ,U100-00-00_0383 ,46039.27,0,102.19,103.57
Observed WS=U100-00-00      ,U100-00-00_0383 ,44920.4 ,0,102.06,103.39
Observed WS=U100-00-00      ,U100-00-00_0383 ,43528.58,0,101.68,102.92
Observed WS=U100-00-00      ,U100-00-00_0383 ,42339.98,0,100.94,102.2
Observed WS=U100-00-00      ,U100-00-00_0383 ,41257.1 ,0,100.1,101.45
Observed WS=U100-00-00      ,U100-00-00_0383 ,40140.33,0,99.61,101.02
Observed WS=U100-00-00      ,U100-00-00_0383 ,39113.75,0,98.76,100.39
Observed WS=U100-00-00      ,U100-00-00_0383 ,38317.03,0,97.6,99.9
DSS Import GetInterval= 0
DSS Import GetPeak= 0
DSS Import FillOption= 0
