HEC-RAS study U100-00-00.prj: U100-00-00

--- U100-00-00.g01 (geometry) --- (continued)

Type RM Length L Ch R = 2 ,102144.1,,,
BEGIN DESCRIPTION:
ROAD NORTH OF MCGILL
END DESCRIPTION:
Node Name=NORTH OF MCGILL
Bridge Culvert--1,0,-1,-1, 0
Deck Dist Width WeirC Skew NumUp NumDn MinLoCord MaxHiCord MaxSubmerge Is_Ogee
15.5,59,2.6,0, 60, 60, , , 0.98, 0, 0,0,,
       0    9.98   29.95   94.83  284.49  294.47  319.43  339.39  349.38   394.3
  414.26  434.22  459.18  469.16  484.13  529.05  554.01  573.97  593.94  608.91
  618.89  633.87  643.85  658.82  688.77  708.73  738.68  753.65  778.61  788.59
  808.56  828.52  863.46  878.43   893.4  913.37  923.35  948.31  963.28  983.24
 1043.14 1058.11 1137.97 1242.78 1332.62 1427.45 1502.32 1602.14 1711.94 1851.69
 2136.19 2265.95 2340.82 2435.65 2500.34 2585.07 2618.58 2631.71 2678.07 2702.58
   151.6  151.86  151.99   151.9  152.09  152.38  151.99  152.26   152.1  152.33
  152.11  152.22  151.94  152.26  151.97     152  151.68   151.9  151.67  151.86
  151.52  151.43  151.68  151.49  151.78  151.67  151.95  151.66   151.9   151.7
  151.95  151.73  151.77  152.04  151.79  152.06  151.81  152.01  151.83  151.99
  151.71  152.04  151.63  151.69  151.36  151.97  152.18  151.84   151.9  151.43
  151.76  151.53  151.05  151.24  150.99   151.3  151.08  151.38  151.18  150.56
       0       0       0       0       0       0       0       0       0       0
       0       0       0       0       0       0       0       0       0       0
       0       0       0       0       0       0       0       0       0       0
       0       0       0       0       0       0       0       0       0       0
       0       0       0       0       0       0       0       0       0       0
       0       0       0       0       0       0       0       0       0       0
       0    9.98   29.95   94.83  284.49  294.47  319.43  339.39  349.38   394.3
  414.26  434.22  459.18  469.16  484.13  529.05  554.01  573.97  593.94  608.91
  618.89  633.87  643.85  658.82  688.77  708.73  738.68  753.65  778.61  788.59
  808.56  828.52  863.46  878.43   893.4  913.37  923.35  948.31  963.28  983.24
 1043.14 1058.11 1137.97 1242.78 1332.62 1427.45 1502.32 1602.14 1711.94 1851.69
 2136.19 2265.95 2340.82 2435.65 2500.34 2585.07 2618.58 2631.71 2678.07 2702.58
   151.6  151.86  151.99   151.9  152.09  152.38  151.99  152.26   152.1  152.33
  152.11  152.22  151.94  152.26  151.97     152  151.68   151.9  151.67  151.86
  151.52  151.43  151.68  151.49  151.78  151.67  151.95  151.66   151.9   151.7
  151.95  151.73  151.77  152.04  151.79  152.06  151.81  152.01  151.83  151.99
  151.71  152.04  151.63  151.69  151.36  151.97  152.18  151.84   151.9  151.43
  151.76  151.53  151.05  151.24  150.99   151.3  151.08  151.38  151.18  150.56
       0       0       0       0       0       0       0       0       0       0
       0       0       0       0       0       0       0       0       0       0
       0       0       0       0       0       0       0       0       0       0
       0       0       0       0       0       0       0       0       0       0
       0       0       0       0       0       0       0       0       0       0
       0       0       0       0       0       0       0       0       0       0
BR Coef=-1 , 0 , 0 ,, 0 ,,,0.8,-1,,0,
WSPro=,,,, 1 ,,,, 0 ,,,, 0 ,,,,-1 ,-1 ,-1 , 0 , 0 , 0 , 0 , 0
Culvert=1,3.5,,59,0.013,0.5,1,1,3,144.19,2652.42,144.45,2652.42,Culvert #1  , 0 ,15.5
Culvert Bottom n=0.013
BC Design=,, 0 ,, 0 ,,,,,,
BC Use User HTab Curves=0
BC User HTab FreeFlow(D)= 0

Type RM Length L Ch R = 1 ,102116.5,360.02,186.18,108.23
BEGIN DESCRIPTION:
Downstream Section - ROAD NORTH OF MCGILL
END DESCRIPTION:
XS GIS Cut Line= 6
3001007.4213943613898730.14923163000762.5432751913896296.8099382
3000748.1768341113896193.36132623000708.9328181113896068.1814584
3000467.7902557713895899.4504967 2998051.983735713890692.0298092
#Sta/Elev= 30
       0   150.4  998.22  151.24 2081.28  149.34 2245.99  150.24 2465.52  149.55
  2545.1  148.21 2575.07  145.24 2614.32  149.17 2650.01   144.4 2682.84  149.49
 2707.51   151.1 2766.62   148.6 2993.21  148.36 5356.36   149.3  5691.1  148.32
 5711.08  144.57 5736.06  150.05 5761.05  150.36 5801.01  148.47 5905.93   148.4
 6635.36  149.94 6990.08  149.23    7100  150.45 7129.97   148.3 7149.96  149.76
 7229.89  149.82 8643.79  149.52 8673.76  148.04 8683.76  150.04 8718.73  148.62
#Mann= 3 , 0 , 0
       0     .07       0 2614.32     .04       0 2682.84     .07       0
#XS Ineff= 3 ,-1
       0 2650.67   150.3 2654.17 5761.05  148.36 5761.05 8718.73   150.5
Permanent Ineff=
       F       F       F
Bank Sta=2614.32,2682.84
XS Rating Curve= 0 ,0
Exp/Cntr=0.5,0.3

Type RM Length L Ch R = 1 ,101930.3,36.99,51.84,24.81
XS GIS Cut Line= 4
3002749.8362166113898164.83277693000898.3546833513895932.7896689
3000579.0685765313895911.42980342998201.5529903613890725.0067773
#Sta/Elev= 30
       0  149.32 1322.72  149.11  1332.7  147.83 1357.66  149.21 1412.56  147.24
 1427.54  148.97 1632.18  150.15 2181.24  148.79 2845.09  150.07    3025  148.29
    3045  150.97 3050.03  149.45  3055.8  145.04 3065.85  145.08 3077.76   149.2
    3095  151.58    3130  148.52    3185  148.22 5932.78  148.37 5957.76  144.28
 5967.75  147.51 6007.72   149.9  6032.7  147.83 7341.62  150.12  7371.6  148.09
 8280.86   149.7  8860.4  148.43 8880.39  149.66 8900.37  147.58 8925.35  150.25
#Mann= 3 ,-1 , 0
       0     .07       0    3045     .04       0    3095     .07       0
#XS Ineff= 2 ,-1
       0    1737  150.19 6007.72 8925.35   149.9
Permanent Ineff=
       F       F
Bank Sta=3045,3095
XS Rating Curve= 0 ,0
Exp/Cntr=0.3,0.1

Type RM Length L Ch R = 1 ,101878.4,35.52,49.78,26.29
Node Name=AF
XS GIS Cut Line= 4
3002751.34179103 13898113.0182483000899.8605858513895880.9748119
3000580.5741509513895859.61527452998230.0785238613890725.9677334
#Sta/Elev= 30
       0  149.24    1158  149.44 1317.73  147.83 1362.65  149.47  1392.6  147.27
 1412.56  149.38  1562.3  150.39 2156.28  148.83  2261.1  150.25 2560.58  149.09
 2590.53  150.55 2954.15  148.28 3042.77  149.63 3064.53  144.42 3072.46  145.47
 3079.95  149.55 3096.92  151.51 3126.46  148.48 5603.38  149.01  5878.2  148.25
 5898.18   144.4 5928.16  149.82 5978.13  147.79 7237.27  148.77 7282.24   150.3
 7307.23  148.32 7382.17  148.19 8821.17  149.67 8846.15  147.61 8866.14  150.03
#Mann= 3 , 0 , 0
       0     .07       0 3042.77     .04       0 3079.95     .07       0
#XS Ineff= 2 ,-1
       0  1562.3  150.39 5928.16 8866.14  149.82
Permanent Ineff=
       F       F
Bank Sta=3042.77,3079.95
XS Rating Curve= 0 ,0
Exp/Cntr=0.3,0.1

Type RM Length L Ch R = 1 ,101828.7,35.9,51,33.12
XS GIS Cut Line= 4
3002752.78798236 13898063.2585053000901.3067771913895831.2153969
3000582.0203422813895809.85585962998267.6755615313890727.3584787
#Sta/Elev= 30
       0  149.33    1345   149.4    1375  147.11    1395  149.27    1455  150.43
 2973.84  149.59 3027.99  148.47 3037.84  149.86 3047.79  149.62  3054.2  146.29
 3063.91   144.6 3087.07  150.96 3101.84  151.11 3116.61  148.41 3170.76   148.2
 4334.92  148.19 4384.92  149.86 5814.81  148.42  5839.8  144.54  5864.8  149.59
  5919.8   147.9  5929.8  149.04  7164.7  149.08  7194.7  150.29  7209.7  148.62
  7224.7  150.01 7249.69  148.18 8764.61  149.52 8779.61  147.47 8804.61  149.88
#Mann= 3 , 0 , 0
       0     .07       0 3037.84     .04       0 3087.07     .07       0
#XS Ineff= 2 ,-1
       0    1455  150.43  5869.8 8804.61  149.73
Permanent Ineff=
       F       F
Bank Sta=3037.84,3087.07
XS Rating Curve= 0 ,0
Exp/Cntr=0.5,0.3

Type RM Length L Ch R = 1 ,101777.7,86.37,125.48,57.07
BEGIN DESCRIPTION:
Upstream Section - DIRT ROAD
END DESCRIPTION:
XS GIS Cut Line= 5
3002754.2696066913898012.27796393000902.7884015313895780.2348558
3000739.6821004513895769.32313233000583.5019666113895758.8749904
2998359.6432253613890790.1736418
#Sta/Elev= 30
       0  149.37    1315  149.58    1360  147.46    1390     150    1415  148.99
    1440  150.37 2040.01  149.48 2090.01  150.66 2135.01  148.94 2180.01  150.74
    2220  149.12 2954.48  148.48 3038.75  149.04  3042.4  151.87 3047.96  149.56
 3054.09  145.95 3061.56   144.6 3078.09  149.34 3092.81  151.66 3117.27  148.74
 3234.99  148.39 5739.35  148.57 5759.34  147.49 5774.34  144.16 5804.33  149.64
 5849.32     148 7039.01  149.04    7069  150.29 7183.97  147.95 8663.61  149.06
#Mann= 3 , 0 , 0
       0     .07       0 3047.96     .04       0 3078.09     .07       0
#XS Ineff= 4 ,-1
       0    1455  150.59 3047.96 3057.56  148.48 3065.56 3078.09  148.26
 5804.33 8663.61  149.64
Permanent Ineff=
       F       F       F       F
Bank Sta=3047.96,3078.09
XS Rating Curve= 0 ,0
Exp/Cntr=0.5,0.3

Type RM Length L Ch R = 2 ,101717.7,,,
BEGIN DESCRIPTION:
DIRT ROAD
U00_1900
END DESCRIPTION:
Node Name=DIRT ROAD
Bridge Culvert--1,0,-1,-1, 0
Deck Dist Width WeirC Skew NumUp NumDn MinLoCord MaxHiCord MaxSubmerge Is_Ogee
55,14.5,2.6,0, 10, 10, , , 0.98, 0, 0,0,,
 2904.95 2919.81 2944.58 2979.25 3004.02 3033.74  3048.6 3063.46 3092.81 3107.49
  148.74  149.39  149.95  150.84  151.52   152.2  151.99   151.7  152.03  151.61
       0       0       0       0       0       0       0       0       0       0
 2904.95 2919.81 2944.58 2979.25 3004.02 3033.74  3048.6 3063.46 3092.81 3107.49
  148.74  149.39  149.95  150.84  151.52   152.2  151.99   151.7  152.03  151.61
       0       0       0       0       0       0       0       0       0       0
BR Coef=-1 , 0 , 0 ,, 0 ,,,0.8,-1,,0,
WSPro=,,,, 1 ,,,, 0 ,,,, 0 ,,,,-1 ,-1 ,-1 , 0 , 0 , 0 , 0 , 0
Culvert=1,8,,29.3,0.013,0.5,1,1,3,143.26,3061.56,143.56,3061.56,Culvert #1  , 0 ,48.4
Culvert Bottom n=0.013
BC Design=,, 0 ,, 0 ,,,,,,
BC Use User HTab Curves=0
BC User HTab FreeFlow(D)= 0

Type RM Length L Ch R = 1 ,101652.2,37.02,49.73,57.65
BEGIN DESCRIPTION:
Downstream Section - DIRT ROAD
END DESCRIPTION:
XS GIS Cut Line= 5
3002757.9149406113897886.85170563000906.4337354513895654.8085975
3000743.3274343613895643.89687393000587.1473005313895633.4487321
2998363.2885592713890664.7473834
#Sta/Elev= 30
       0  149.28    1255  148.76    1285  150.09    1325  147.82    1385  149.83
    1495  150.21    2320  148.97    2400  149.98    2435  148.74    2765  148.78
    2785  147.55 3013.93  148.63 3051.15  147.62 3060.93  144.65 3069.22  145.97
 3076.05  149.69 3092.81  151.97 3117.27  149.18 3141.73  148.54 5614.38  148.49
 5634.37   144.3 5659.37  149.64 5709.35  147.99 6829.06  149.99 7014.01  149.86
 7039.01  148.05 8478.65  149.74 8553.63  149.36 8568.63  147.45 8663.61   149.6
#Mann= 3 , 0 , 0
       0     .07       0 3013.93     .04       0 3076.05     .07       0
#XS Ineff= 4 ,-1
       0    1495  150.21 3013.93 3057.56  148.16 3065.56 3076.05  148.16
 5669.36 8663.61  149.67
Permanent Ineff=
       F       F       F       F
Bank Sta=3013.93,3076.05
XS Rating Curve= 0 ,0
Exp/Cntr=0.5,0.3

Type RM Length L Ch R = 1 ,101602.5,37.36,50.18,20.44
XS GIS Cut Line= 4
3002759.3594915313897837.13986283000907.8782863613895605.0967547
3000588.5918514413895583.73721742998577.4406900313890737.9437594
#Sta/Elev= 30
       0  149.42    1235  148.57    1280  150.22    1320  147.65    1350  149.75
    1475  150.13    2430   149.9    2720  147.59 2998.46  148.81 3047.69  148.09
 3062.61  144.53 3068.07  145.13    3075  148.92 3091.99  152.09 3131.38   148.7
 3264.97  148.29 5333.59  148.69 5518.46  148.27 5548.44  144.32 5573.42  149.56
 5618.39  148.25 5663.36  149.42 6008.13   148.2 6907.52  150.03  6937.5  148.01
 7047.42  149.89 8216.63  149.18  8416.5  150.43 8441.49  148.01 8466.47  150.23
#Mann= 3 , 0 , 0
       0     .07       0 2998.46     .04       0    3075     .07       0
#XS Ineff= 2 ,-1
       0    1475  150.27 5583.42 8466.47  149.83
Permanent Ineff=
       F       F
Bank Sta=2998.46,3075
XS Rating Curve= 0 ,0
Exp/Cntr=0.3,0.1

Type RM Length L Ch R = 1 ,101552.3,36.62,48.97,27.34
XS GIS Cut Line= 4
3002760.8174938613897786.96935943000909.3362886913895554.9262514
3000590.04985377 13895533.5667142998595.97313328 13890739.095988
#Sta/Elev= 30
       0  149.35    1220  148.51    1265  150.09    1315   147.7    1355  150.07
 1810.01  148.91 2160.01   150.2    2380  148.66    2410  149.96    2655  147.66
    2680  148.91 2998.46  148.96 3048.86  148.13 3060.78  144.27 3075.64     149
 3091.99  152.17 3111.69  149.48 3141.23  148.51 3334.94   148.1    5354  148.47
 5473.94   147.9 5488.93  144.19 5518.92  149.46 5988.69  148.29 6858.27  150.06
 6878.26  148.22  6993.2  149.76 8377.55  149.84 8392.54  147.59 8412.53  150.64
#Mann= 3 , 0 , 0
       0     .07       0 2998.46     .04       0 3075.64     .07       0
#XS Ineff= 2 ,-1
       0    1635  150.21 5528.91 8412.53  149.72
Permanent Ineff=
       F       F
Bank Sta=2998.46,3075.64
XS Rating Curve= 0 ,0
Exp/Cntr=0.3,0.1

Type RM Length L Ch R = 1 ,101503.3,747.48,921.12,413.23
XS GIS Cut Line= 4
3002762.2403912813897738.0081713 3000910.759186113895505.9650632
 3000591.472751213895484.60519782998649.3437614413890740.6005782
#Sta/Elev= 30
       0  149.21    1190  149.96    1225  148.26    1275  149.86    1315  147.46
    1350  149.88    1625   150.7 1790.01  149.17    2370  149.78    2405  148.26
    2420  149.34    2640   147.8 3013.23  148.64 3047.69  147.72 3063.02  144.31
  3075.6  148.64 3091.99  151.96 3131.38   148.5 5333.41  148.59 5413.35  147.86
 5433.33  144.24 5448.32  148.26 5463.31   149.4 5937.95  148.17 6792.31  149.95
 6822.29  148.38 6847.27   149.9 8306.17  150.39 8326.16  147.85 8346.14  150.51
#Mann= 3 , 0 , 0
       0     .07       0 3013.23     .04       0  3075.6     .07       0
#XS Ineff= 2 ,-1
       0    1745  150.21 5568.23 8346.14  149.51
Permanent Ineff=
       F       F
Bank Sta=3013.23,3075.6
XS Rating Curve= 0 ,0
Exp/Cntr=0.3,0.1

Type RM Length L Ch R = 1 ,100582.2,665.75,1050.88,808.34
XS GIS Cut Line= 5
3003046.2234191113897171.74978943000833.1799449513894577.2700702
3000697.7901238713894570.29993982999339.4624599413892185.3909957
2998770.3907634513890744.0680909
#Sta/Elev= 30
       0  149.03 1353.06  149.16 1422.96  149.03 1447.93  147.28 1492.86  149.68
 1592.72  148.41 1667.61  149.89 1842.37  147.38 3414.94   148.4 3448.84  147.35
 3462.55  143.59 3480.84   148.7 3492.41   150.9 3516.62  148.42 3560.67  147.76
 4695.53  148.27 4820.51  147.51 4840.51  144.65 4855.51  148.39 4880.51  150.14
  4915.5  148.22  4930.5  149.45 5620.42  147.74 6270.35  150.11 6325.34  148.49
 6365.33  150.19 7680.01  148.87 7799.98  150.16 7814.97  146.48 7839.97   150.8
#Mann= 3 , 0 , 0
       0     .07       0 3414.94     .04       0 3480.84     .07       0
#XS Ineff= 2 ,-1
       0 1667.61  149.89 4880.51 7839.97  150.14
Permanent Ineff=
       F       F
Bank Sta=3414.94,3480.84
XS Rating Curve= 0 ,0
Exp/Cntr=0.3,0.1

Type RM Length L Ch R = 1 ,99531.3 ,22.18,41.16,78.09
BEGIN DESCRIPTION:
Channel data copied from RS 99490.14 to avoid lateral channel
END DESCRIPTION:
XS GIS Cut Line= 5
3003428.9195041113897018.20678943000868.0601245313893574.4699104
3000758.0701870313893479.47895873000103.3513521113892206.2242873
2999358.9145207713890764.4361604
#Sta/Elev= 30
       0  148.48  774.38  149.52 1533.77  147.29 1568.74  148.83 1583.72  146.67
 1628.69  148.13  1738.6   146.6 1778.57  148.58 1803.55  146.95 4296.36  148.01
 4310.47 146.687    4318 143.007  4322.5 142.877 4356.49 148.757 4417.47   149.9
 4441.83  144.26 4451.81  144.95 4461.79   148.5 4481.74  149.75 4536.61  147.49
 5090.34  148.99 5659.03  147.72 5863.56  149.67 5893.51  147.77 5913.48  149.05
 7286.46  148.56 7416.26  149.13 7446.22  150.63 7471.18  147.31 7491.15  150.37
#Mann= 3 , 0 , 0
       0     .07       0 4296.36     .04       0 4356.49     .07       0
#XS Ineff= 2 ,-1
       0  774.38  149.52 5863.56 7491.15  149.67
Permanent Ineff=
       F       F
Bank Sta=4296.36,4356.49
XS Rating Curve= 0 ,0
Exp/Cntr=0.3,0.1

Type RM Length L Ch R = 1 ,99490.14,389.02,855.6,849.62
XS GIS Cut Line= 6
3003444.96835652  13897006.272433000882.7969716913893560.7707908
3000887.7329854413893480.19385233000932.2483163613892233.3101912
3000967.0195722713892168.90907333001051.3448629413890815.4865833
#Sta/Elev= 30
       0  148.58  609.82  149.64 1499.56  148.55 1519.56  147.23 1549.55  149.18
 1574.54  146.47 1594.54  147.98 1744.49  147.27 1769.48  148.58 1824.47  146.74
 1854.46     148 4268.76  148.01 4283.76  147.61 4290.47  146.54    4298  142.86
  4302.5  142.73    4327  147.55 4350.74  149.34 4355.49  149.85 4404.43  154.26
 4429.38  153.61 4464.32  150.37 5153.04  151.32 5944.63  150.89 6159.01  148.39
 6622.66  146.22 6672.52  147.63 6702.43  149.76  6986.6  148.13 7051.42  148.86
#Mann= 3 ,-1 , 0
       0     .07       0 4268.76     .04       0 4355.49     .07       0
#XS Ineff= 1 ,-1
       0  829.76  149.56
Permanent Ineff=
       F
#Block Obstruct= 2 , 0
       0                 4464.32       0  150.37
Bank Sta=4268.76,4350.74
XS Rating Curve= 0 ,0
Exp/Cntr=0.3,0.1

Type RM Length L Ch R = 1 ,98634.54,1013.93,1139,1156.61
Node Name=AE
XS GIS Cut Line= 4
 3003793.5998771 13896896.6466653001921.9992896213894308.4969857
3001742.0898725213893618.37008513001730.8198819513893515.0300687
#Sta/Elev= 30
       0  148.88  339.89  148.89  404.87  147.34  429.86  149.07 1169.62  149.04
 1329.57  148.44 1349.56  146.53 1364.56  149.07 1384.55  149.56 1399.55  147.18
 1419.54  148.32 1659.46  147.29 1979.36  147.97 1989.35  147.04 2029.34  148.58
 2059.33   146.6 2079.32  147.66  2139.3  147.75 3098.99  146.86 3902.16  147.86
  3930.7  146.48 3938.36  142.12 3942.94  142.06 3947.67  142.57 3952.34  144.99
 3978.61  148.88  3981.4  149.64  3991.3  154.02 3996.25  154.97  4011.1  153.36
#Mann= 3 ,-1 , 0
       0     .07       0 3902.16     .04       0  3981.4     .07       0
#XS Ineff= 1 ,-1
       0 1384.55  149.56
Permanent Ineff=
       F
Bank Sta=3902.16,3978.61
XS Rating Curve= 0 ,0
Exp/Cntr=0.3,0.1

Type RM Length L Ch R = 1 ,97495.54,914.46,724.04,697.53
XS GIS Cut Line= 4
3004004.6119222813896936.55570593002969.7547400313894241.7103738
3002873.2998804513893662.91002233002879.1400918713893573.2300835
#Sta/Elev= 30
       0  148.95  993.87  148.54 1093.75  148.41  1143.7  147.49 1183.65  148.33
 1198.63   146.6 1208.62  148.45 1218.61  148.91 1233.59  146.82 1248.58  147.76
 1288.53  148.09 1523.26  148.78 1767.98  148.45 2002.71  146.52 2467.18  148.42
 2512.13  147.76 2522.12   146.6 2567.07  148.93 2622.01  145.77 2656.97  147.49
 2686.93  147.61 3468.52  147.75 3488.47  147.02 3495.43     146 3504.98  141.64
  3512.2  141.85 3544.61  146.53 3548.53   148.6 3558.37  153.11 3563.37  153.96
#Mann= 3 ,-1 , 0
       0     .07       0 3468.52     .04       0 3548.53     .07       0
#XS Ineff= 1 ,-1
       0 1218.61  148.91
Permanent Ineff=
       F
Bank Sta=3468.52,3548.53
XS Rating Curve= 0 ,0
Exp/Cntr=0.3,0.1

Type RM Length L Ch R = 1 ,96771.5 ,329.29,362.48,360.57
XS GIS Cut Line= 5
3004358.7975656113897021.56012913003981.40002644 13894371.009984
3003627.2199605313893742.33998153003591.8000838613893644.9399139
 3003468.216669613893505.1915057
#Sta/Elev= 30
       0  148.72   884.1  148.41  1178.8   147.8 1233.75  146.27 2687.24  147.66
 2766.86  146.15 2831.55  148.45 2866.39  145.76 2891.27  149.19 2911.18  147.21
 3269.47   147.7 3289.38  145.13 3299.33  147.34 3314.26   147.7  3349.1  145.56
 3388.91  147.95 3408.73  147.22 3458.08  148.28    3480  146.46 3498.29  140.18
 3533.97  146.18 3541.78  148.61 3551.59  150.55 3571.23  150.96 3595.78   150.3
 3610.51  147.71 3635.06  147.09 3664.51  149.48 3679.24  152.81 3689.06  153.62
#Mann= 3 ,-1 , 0
       0     .07       0 3458.08     .04       0 3541.78     .07       0
#XS Ineff= 1 ,-1
       0  779.21   148.5
Permanent Ineff=
       F
Bank Sta=3458.08,3541.78
XS Rating Curve= 0 ,0
Exp/Cntr=0.3,0.1

Type RM Length L Ch R = 1 ,96356.5 ,22.07,25,25.87
BEGIN DESCRIPTION:
Updated (March 2016)
END DESCRIPTION:
XS GIS Cut Line= 6
     3004408.113     13897013.34     3004208.497     13893952.59
     3004194.866     13893900.97     3004119.841     13893719.31
     3003578.938     13893069.89     3003493.052     13892994.15
#Sta/Elev= 30
       0  148.54 1133.98  147.77 1178.94  146.25 1193.93  147.32 1208.92  146.12
 2372.88  147.12 2802.49  146.26 3002.31  147.67 3032.29  145.96 3062.26  146.88
 3091.52  142.87 3135.39  140.71 3253.31  141.18 3327.16  146.02 3573.93  145.71
 3680.82  148.15 3691.15  147.98 3713.82  146.45 3728.57   140.9 3743.33  140.92
 3749.68  142.35 3778.18  147.87  3795.8  148.75 3967.51  148.64 4037.46  147.04
 4182.29  147.98  4227.1  146.86 4242.03  148.11 4256.97  152.26 4276.89  153.62
#Mann= 6 ,-1 , 0
       0     .07       0 3002.31     .07       0 3680.82     .04       0
 3728.57    .035       0 3749.68     .04       0 3778.18     .07       0
#XS Ineff= 1 ,-1
    3968    4276   148.6
Permanent Ineff=
       F
#Block Obstruct= 1 ,-1
 3047.27 3638.69  146.87
Bank Sta=3691.15,3778.18
XS Rating Curve= 0 ,0
Exp/Cntr=0.3,0.1

Type RM Length L Ch R = 1 ,96331.5 ,58.27,66,68.31
BEGIN DESCRIPTION:
Updated (March 2016)
END DESCRIPTION:
XS GIS Cut Line= 6
     3004410.884     13897012.88     3004220.632     13893925.75
     3004206.597     13893873.78     3004137.778     13893704.37
     3003624.707      13893085.5     3003494.448     13892965.44
#Sta/Elev= 30
       0   148.5 1109.43  147.69 1124.42  146.85 1154.41  147.37  1169.4  146.28
 1189.39  147.33 1204.38  146.43 2413.75  147.21 2803.55  146.26 2983.46  147.26
 3013.44  146.25 3043.43  146.75 3088.19  140.77 3156.71  140.76 3196.27  141.45
 3260.56  146.52 3329.79  145.84 3369.35  148.02 3670.59  147.27 3738.85  141.77
 3864.25  147.11 3870.43  148.77 3925.05  148.75 4049.19  146.78 4193.35   146.6
 4208.05  148.25 4257.02  146.71 4271.72  147.76 4301.11  153.68  4310.9   153.7
#Mann= 3 ,-1 , 0
       0     .07       0 3670.59    .015       0 3864.25     .07       0
#XS Ineff= 1 ,-1
    3924    4310   148.7
Permanent Ineff=
       F
#Block Obstruct= 1 ,-1
 3043.43 3354.51  146.75
Bank Sta=3670.59,3864.25
XS Rating Curve= 0 ,0
Exp/Cntr=0.3,0.1

Type RM Length L Ch R = 1 ,96265.5 ,35.31,40,41.4
BEGIN DESCRIPTION:
Updated (March 2016)
END DESCRIPTION:
XS GIS Cut Line= 6
     3004418.198     13897011.66     3004252.629     13893854.79
     3004237.528     13893801.89     3004173.715     13893637.84
     3003776.278     13893163.83     3003500.853     13892831.25
#Sta/Elev= 30
       0  148.43 1128.57  147.98 1173.51  146.36 1188.49  147.38 1438.18  146.24
 2736.53  146.24 2946.27  147.27 2961.25  146.12 2986.22   146.8 3031.16  141.48
  3076.1  140.62 3106.07  141.76 3136.03   146.3    3175  145.99 3202.51  147.57
 3397.19     147    3400     149    3500     149    3512     147 3524.95  146.84
 3708.62  147.09 3778.38  141.08 3908.57  147.07 3916.67  148.77  3936.5  149.03
 4045.62  146.69 4378.17   147.1 4393.06   147.3  4427.8  152.64 4442.69  153.32
#Mann= 3 ,-1 , 0
       0     .07       0 3708.62    .015       0 3908.57     .07       0
#XS Ineff= 2 ,-1
       0    1128   147.9    3983    4442   148.7
Permanent Ineff=
       F       F
#Block Obstruct= 1 ,-1
 2986.22 3151.01  146.65
Bank Sta=3708.62,3908.57
XS Rating Curve= 0 ,0
Exp/Cntr=0.3,0.1

Type RM Length L Ch R = 1 ,96225.5 ,195.14,221.04,228.76
BEGIN DESCRIPTION:
Updated (March 2016)
END DESCRIPTION:
XS GIS Cut Line= 6
     3004422.631     13897010.92     3004273.875      13893822.8
     3004271.966     13893811.62     3004256.219     13893758.16
     3004198.528     13893605.94     3003503.042     13892775.55
#Sta/Elev= 30
       0  148.44  1118.8  147.63 1168.75  146.19 1183.73  147.34 2127.72  146.07
 2921.88  146.91 2966.83  146.63  2996.8  141.96 3011.78  141.09 3056.73  140.88
 3076.71  142.11 3106.68  146.71 3254.02  147.08 3298.13     149    3530     149
 3543.09  147.53 3580.51  146.48 3610.74  137.54 3891.49  135.85 3903.82  138.09
  3929.3  134.86 3967.72     136 4231.44  135.65 4287.34  138.95 4369.03  146.81
 4385.24  146.92 4444.73  146.78 4474.68  149.22 4489.65  153.39 4504.63   153.7
#Mann= 3 ,-1 , 0
       0     .07       0 3543.09     .04       0 4385.24     .07       0
#XS Ineff= 2 , 0
       0                    3787       0  146.92
Permanent Ineff=
       F       F
#Block Obstruct= 1 ,-1
 2966.83 3106.68  146.63
Bank Sta=3543.09,4385.24
XS Rating Curve= 0 ,0
Exp/Cntr=0.3,0.1

Type RM Length L Ch R = 1 ,96004.46,649.07,460.08,554.16
BEGIN DESCRIPTION:
Updated (March 2016)
END DESCRIPTION:
Node Name=AD
XS GIS Cut Line= 5
3004443.8023168613897007.39283463004368.1617201113893616.8960067
 3004221.430058213893179.41984753004060.5901567813893044.9001034
3003511.0253110213892624.3222044
#Sta/Elev= 30
       0  148.43 1098.81  147.15  1108.8  148.14 1163.74  146.16 1183.72  147.59
 1198.71  146.41 2082.75  147.27 2816.95  145.78 2846.92  146.82 2886.88  141.19
 2906.85   140.8 2951.81  142.12 2981.77  146.76    3145     149    3720     149
 3731.89  147.84 3782.74  142.42 3806.22  141.87 3851.96  135.21 4012.02  131.98
 4016.25  134.36 4224.62  138.09 4559.47   134.6 4599.39  141.89 4623.92  142.44
 4656.49  147.78 4709.68  146.95 4729.59  149.61 4739.55  152.54 4754.48   153.4
#Mann= 3 ,-1 , 0
       0     .07       0 3731.89     .04       0 4656.49     .07       0
#XS Ineff= 1 ,-1
       0 1733.13  147.09
Permanent Ineff=
       F
#Block Obstruct= 1 ,-1
 2846.92 2981.77  145.82
Bank Sta=3731.89,4656.49
XS Rating Curve= 0 ,0
Exp/Cntr=0.3,0.1

Type RM Length L Ch R = 1 ,95544.38,125.59,110.94,131.34
BEGIN DESCRIPTION:
Updated (March 2016)
END DESCRIPTION:
XS GIS Cut Line= 6
3004514.6394455313896979.05791753004649.2300556213893281.3579638
3004417.3699550313892764.37015273004134.6999166913892332.0501512
3003795.4991515313891804.88946013003679.4367196113891746.3557845
#Sta/Elev= 30
       0  148.17 1118.53  147.62 1133.51  146.08  1148.5  147.78 1173.46  145.88
 1183.45  147.04 1847.57   147.6 2501.71  147.14 2516.69  145.98 2541.66  147.39
 2596.58  141.12 2631.54  141.02 2651.51  142.72 2671.48   146.9 2851.25  147.43
    2888     149    4050     149 4073.81  147.55 4145.28  144.37 4217.89  134.34
 4269.99  131.68 4319.35  147.29    4705     149 4862.85  147.93 4982.26   150.2
 5061.86  150.27 5235.99  147.09 5360.37  150.02 5420.12  147.12 5540.11  148.77
#Mann= 4 ,-1 , 0
       0     .07       0    2888     .05       0 4073.81     .04       0
 4319.35     .07       0
#XS Ineff= 3 ,-1
       0 1847.57   147.6                         4708.75 5540.11  148.83
Permanent Ineff=
       F       F       F
#Block Obstruct= 1 ,-1
 2541.66 2686.46  146.17
Bank Sta=4073.81,4319.35
XS Rating Curve= 0 ,0
Exp/Cntr=0.3,0.1

Type RM Length L Ch R = 1 ,95444.3 ,648.25,533.1,582.79
BEGIN DESCRIPTION:
Updated (March 2016)
END DESCRIPTION:
XS GIS Cut Line= 6
     3004523.591      13896975.7     3004686.167      13893492.6
     3004734.683     13893228.28     3004419.891     13892513.88
     3003798.269     13891471.72       3003689.4      13891395.8
#Sta/Elev= 30
       0  148.12 1048.36  148.17 1108.26  147.98 1123.24  146.28 1143.21  147.79
 1173.16  146.31  2460.6  147.64 2520.39  146.58 2535.34  143.27 2550.29  141.78
 2580.18  140.79 2615.06  142.72 2644.95  147.47 2854.21  147.74    2875     149
    4200     149 4210.12  147.56  4238.6  146.64  4339.2  131.53 4355.69  131.43
 4379.89  133.84 4436.55  146.84    4475     148    4765     149 4900.13  146.82
 5233.46  150.17 5501.59  147.23 5605.86  148.81 5739.92  146.99 5882.58  148.92
#Mann= 3 ,-1 , 0
       0     .07       0 4210.12     .04       0 4436.55     .07       0
#Block Obstruct= 1 ,-1
 2505.44 2692.83  147.07
Bank Sta=4210.12,4436.55
XS Rating Curve= 0 ,0
Exp/Cntr=0.3,0.1

Type RM Length L Ch R = 1 ,94911.28,396.93,394.92,443.22
BEGIN DESCRIPTION:
Updated (March 2016)
END DESCRIPTION:
XS GIS Cut Line= 6
3004571.3089516213896957.80664773004748.4021013513894067.6506826
 3005153.770713213893061.54606753005029.2899910213892642.9199363
3004962.2701119513892443.08011293003742.5143493613889526.9885041
#Sta/Elev= 30
       0  147.88 1008.46  148.38 1108.31   146.1 1128.28  147.84 1148.25  146.49
 1198.17  147.74 2051.87  146.57    2360   148.1    4075     149 4140.41  147.67
 4285.58  146.52 4339.78  133.95 4632.17  133.48 4660.84  130.89 4668.41  130.97
 4728.27  145.35  4750.5  146.29  5087.2  147.89 5132.14  140.81 5446.73  139.67
 5481.69  139.84 5571.57  149.88 5661.45  146.45 5821.24  149.28 5916.12  146.48
 6480.38  149.37 6819.94  146.98 6974.74  149.35 7009.69  145.45 7788.68  146.11
#Mann= 5 ,-1 , 0
       0     .07       0    2360     .04       0 4140.41     .07       0
 4285.58     .04       0  4750.5     .07       0
#XS Ineff= 2 ,-1
       0 2331.44  147.46  5087.2 7788.68  147.89
Permanent Ineff=
       F       F
#Block Obstruct= 2 ,-1
 2391.35 2521.15   146.3  5087.2  5546.6  146.89
Bank Sta=4285.58,4750.5
XS Rating Curve= 0 ,0
Exp/Cntr=0.3,0.1

Type RM Length L Ch R = 1 ,94516.37,62.9,63.84,107.48
BEGIN DESCRIPTION:
Updated (March 2016)
END DESCRIPTION:
XS GIS Cut Line= 6
3004621.5142317713897013.08114343004690.2857477813895095.8162772
3005394.6721342813893218.14713233005398.8401049413892493.1249603
3005204.6000078613891756.87938553005125.2418988613890767.5965872
#Sta/Elev= 30
       0  148.15 1059.17  148.22 1159.09  146.16 1254.02  147.95 2053.06  146.23
 2325.28   148.2 2380.86  146.93 2400.62  142.25 2430.26  141.65 2464.84  146.98
 2499.42  147.63 2910.93   146.1    2975     149    4175     149    4195     147
 4669.07  145.55 4743.26  132.99 4774.81  129.91 4899.43  136.22 4935.66  143.79
 4971.41  147.25 5392.87  147.32 5421.88  149.26 5576.43  146.66 5720.93  148.88
  5825.8  146.03 5915.57  148.28 6050.23  148.64 6130.02  145.68 6424.27  147.63
#Mann= 6 ,-1 , 0
       0     .07       0 2325.28     .05       0 4669.07     .04       0
 4971.41     .07       0 5392.87     .15       0 5720.93     .07       0
#XS Ineff= 3 ,-1
       0 4436.07  146.88 5110.99 6050.23  146.73 6050.23 6424.27  147.74
Permanent Ineff=
       F       F       F
#Block Obstruct= 1 ,-1
 2380.86 2464.84  145.93
Bank Sta=4669.07,4971.41
XS Rating Curve= 0 ,0
Exp/Cntr=0.3,0.1

Type RM Length L Ch R = 1 ,94452.52,51.42,56.4,96
BEGIN DESCRIPTION:
Updated (March 2016)
END DESCRIPTION:
XS GIS Cut Line= 6
3004641.1250849413896989.12515463004732.1249029513895073.1250496
3004802.1250910313894746.12504743005320.1250392813893756.1250589
3005446.1251153613893277.12503273005398.17836086 13891017.241101
#Sta/Elev= 30
       0  148.09 1014.03   146.9 1029.01  148.29 1123.92  147.57 1133.91  145.95
  1148.9  147.68 1203.85  146.22 1228.82   147.9 2117.81  146.62 2479.17  147.72
  2920.5  145.91    2950     149    4159     149    4260   146.8 4675.21  146.61
  4746.2  129.52 4761.75  130.15 4813.17  139.61 4901.51  136.46 4977.52  146.36
    5000     148    5250     148 5271.09  145.86 5291.04  147.86 5362.69  147.48
 5425.44  148.95 5726.19  149.09 5952.06  145.51 6121.16  145.72 6141.06  147.77
#Mann= 5 ,-1 , 0
       0     .07       0 4675.21     .04       0 4977.52     .07       0
 5362.69     .15       0 5726.19     .07       0
#XS Ineff= 4 ,-1
       0 2955.17  147.23 2955.17 4159.06  146.88 5155.88 5753.11  146.43
 5753.11 6141.06   148.8
Permanent Ineff=
       F       F       F       F
Bank Sta=4675.21,4977.52
XS Rating Curve= 0 ,0
Exp/Cntr=0.5,0.3

Type RM Length L Ch R = 1 ,94396.13,178.17,183.98,163.51
BEGIN DESCRIPTION:
Upstream Section - FRY ROAD (Updated March 2016)
END DESCRIPTION:
XS GIS Cut Line= 6
3004665.1250369413896981.12484253004754.1248589513895064.1250676
3004930.1251631113894466.12495133005422.1251633613893504.1249068
3005484.1250393513891772.12508993005606.1251234413891107.1251076
#Sta/Elev= 30
       0  147.94 1004.51  146.91 1014.51  148.08 1109.46   147.6 1124.45  145.44
 1139.44  147.62 1174.43  147.88 1199.42  146.31  1224.4  147.67 2307.07  147.77
 2872.01  145.31 2941.24   147.2 2951.12  145.59 3010.44  144.86 4075.34  146.84
 4404.39  145.21 4647.07  145.59 4678.47  147.26 4715.13   138.8 4741.92  129.94
 4757.89  129.91 4828.64  146.49 5121.56  143.72 5250.56  145.18  5284.8  147.21
 5343.72   146.8 5411.49  145.52 5864.41  144.72 5972.28  146.71  6043.2  147.71
#Mann= 6 ,-1 , 0
       0     .07       0 4678.47     .04       0 4828.64     .07       0
 5343.72     .15       0 5411.49     .07       0 5972.28     .15       0
#XS Ineff= 3 ,-1
       0 2941.24   147.2 2941.24 4708.05  146.88 4829.99  6043.2  146.13
Permanent Ineff=
       F       F       F
Bank Sta=4678.47,4828.64
XS Rating Curve= 0 ,0
Exp/Cntr=0.5,0.3

Type RM Length L Ch R = 3 ,94315.28,,,
BEGIN DESCRIPTION:
FRY ROAD
U00_1800
END DESCRIPTION:
Node Name=FRY ROAD
Bridge Culvert--1,0,-1,-1, 0
Deck Dist Width WeirC Skew NumUp NumDn MinLoCord MaxHiCord MaxSubmerge Is_Ogee
32,106,2.6,0, 60, 60, , , 0.98, 0, 0,0,,
       0  259.76  409.62  554.49  619.43  854.22 1019.07 1098.99 1243.86 1398.72
  1533.6 1818.34  1858.3 2073.05 2430.64 2653.29  2787.1  2831.7 2851.52 2866.39
 2896.06 2910.88 2945.45 2994.83 3152.68 3417.97 3560.67 3653.65 3721.13 4031.46
 4084.72 4159.09 4179.09 4214.09 4234.09 4294.09 4424.09 4553.97 4602.82 4651.66
 4705.38 4708.05 4744.45 4829.99 4833.53 4838.49 4863.29 4893.06 5017.09 5101.43
 5318.12 5322.92 5410.96 5545.52 5595.44 5684.85 5763.12    5806 5951.99 6042.89
  149.85  149.65  149.84  149.59  149.83  149.62   149.9  149.57  149.79  149.52
  149.77  149.27  149.51  148.92  148.91  148.21  148.16  148.38  148.11  147.55
  147.55  148.14  148.37  147.97  147.73  147.68  147.97  147.82  148.11  148.06
  148.33  148.02  147.18  146.88  147.64  147.92  147.93  149.08  150.22  150.85
  153.97  154.02  154.07  154.19  152.96  150.75   150.9  150.51  147.99  146.97
  147.05  146.76  146.89  146.51  146.72  146.31  146.59  146.24  146.13  146.33
       0       0       0       0       0       0       0       0       0       0
       0       0       0       0       0       0       0       0       0       0
       0       0       0       0       0       0       0       0       0       0
       0       0       0       0       0       0       0       0       0       0
       0  148.15  148.02  148.34       0       0       0       0       0       0
       0       0       0       0       0       0       0       0       0       0
       0  259.76  409.62  554.49  619.43  854.22 1019.07 1098.99 1243.86 1398.72
  1533.6 1818.34  1858.3 2073.05 2430.64 2653.29  2787.1  2831.7 2851.52 2866.39
 2896.06 2910.88 2945.45 2994.83 3152.68 3417.97 3560.67 3653.65 3721.13 4031.46
 4084.72 4159.09 4179.09 4214.09 4234.09 4454.09 4568.63 4602.82    4637 4671.19
 4685.85 4691.61  4729.8 4814.75  4823.6 4853.37 4863.29 4893.06 5046.86  5131.2
 5337.32 5356.52 5410.96 5545.52 5595.44 5684.85 5763.12    5806 5951.99 6042.89
  149.85  149.65  149.84  149.59  149.83  149.62   149.9  149.57  149.79  149.52
  149.77  149.27  149.51  148.92  148.91  148.21  148.16  148.38  148.11  147.55
  147.55  148.14  148.37  147.97  147.73  147.68  147.97  147.82  148.11  148.06
  148.33  148.02  147.18  146.88  147.64  147.98     149  149.75  151.05  153.13
  153.41  153.44  153.63  154.06  153.38  151.07  150.78  150.84  147.87  146.89
  147.05  146.76  146.89  146.51  146.72  146.31  146.59  146.24  146.13  146.33
       0       0       0       0       0       0       0       0       0       0
       0       0       0       0       0       0       0       0       0       0
       0       0       0       0       0       0       0       0       0       0
       0       0       0       0       0       0       0       0       0       0
       0  147.79  148.29  148.11       0       0       0       0       0       0
       0       0       0       0       0       0       0       0       0       0
Pier Skew, UpSta & Num, DnSta & Num=  ,4747.05, 2 ,4729.27, 2 , 0 , 0 , 0 ,,
     1.4     1.4
     138     149
     1.4     1.4
     138     149
Pier Skew, UpSta & Num, DnSta & Num=  ,4792.3, 2 ,4774.28, 2 , 0 , 0 , 0 ,,
     1.4     1.4
     138     149
     1.4     1.4
     138     149
Abutment Skew #Up #Dn= , 2 , 2
 4706.06 4729.32
  148.07  139.83
 4690.67 4715.83
  148.21  139.91
Abutment Skew #Up #Dn= , 2 , 3
 4805.77 4831.06
  139.91  148.22
 4793.11 4814.71 4814.91
  140.03 148.115 148.115
BR Coef=-1 , 1 , 1 ,1.25, 0 ,,,0.8,-1,2,0,
WSPro=,,,, 1 ,,,, 0 ,,,, 0 ,,,,-1 ,-1 ,-1 , 0 , 0 , 0 , 0 , 0
BC Design=,, 0 ,, 0 ,,,,,,
BC Use User HTab Curves=0
BC User HTab FreeFlow(D)= 0

Type RM Length L Ch R = 1 ,94212.15,99.25,63.66,20.93
BEGIN DESCRIPTION:
Downstream Section - FRY ROAD (Updated March 2016)
END DESCRIPTION:
XS GIS Cut Line= 6
3004912.1248710313896915.12497453004958.1251071113894997.1248735
3005120.1251111913894395.12509333005590.1251554513893422.1250708
3005648.1250394413891689.12492783005870.1249235313891064.1248655
#Sta/Elev= 30
       0  148.01  484.63  146.93  814.38  147.56  894.32   146.8 1428.92  147.71
 1883.58  146.79 2008.28   147.6 2792.51  145.38 2802.46  147.01 2822.35  147.35
 2837.27  145.25 3726.25  146.35 4349.41  145.98 4504.41  145.01 4578.72  145.12
 4661.89  146.26  4676.4  147.26 4681.47  146.59 4738.44  130.27 4758.17  133.82
 4778.46  135.29 4811.22   145.7 4818.87  146.26 4928.11  144.48 4977.72   145.3
 5141.44  144.23 5416.26  144.25 5893.84  145.43 6015.77  146.68  6042.7  147.02
#Mann= 4 ,-1 , 0
       0     .07       0 4681.47     .04       0 4818.87     .07       0
 6015.77     .15       0
#XS Ineff= 3 ,-1
       0 2822.35     147 2822.35 4691.93  146.38 4818.96  6042.7  146.13
Permanent Ineff=
       F       F       F
Bank Sta=4681.47,4818.87
XS Rating Curve= 0 ,0
Exp/Cntr=0.5,0.3

Type RM Length L Ch R = 1 ,94148.49,94.99,98.61,96.51
BEGIN DESCRIPTION:
Updated (March 2016)
END DESCRIPTION:
XS GIS Cut Line= 6
3005639.2372619513896786.47234473005821.6735768613894283.2598314
3005742.8663197813892329.5685288 3005667.507874713891778.0312461
3005724.2052678613891403.2360639 3005875.007459713891069.1468371
#Sta/Elev= 30
       0   147.5  579.97  146.17 1725.96   147.9 2248.73   145.3 2373.77  147.86
 2464.85  145.97 2479.85  144.39 2496.25  145.98 2534.83  146.87 2630.49  144.77
 2999.51  145.49    3000   147.7    3800   147.7    3890   146.7    3900  144.75
 4282.62  144.06 4342.58  134.14 4503.96  133.81 4541.89  130.04 4579.79  141.59
 4602.35  145.64 4703.01  146.31 4725.31     148    5200   148.4 5236.56  144.61
 5340.23  146.04 5434.03  144.66  5493.3  147.45    5735  147.13 5788.71  146.93
#Mann= 6 ,-1 , 0
       0     .07       0 2496.25     .12       0 2630.49     .07       0
 4282.62     .04       0 4602.35     .07       0    5735     .15       0
#XS Ineff= 4 ,-1
       0 2534.83  146.87                         4709.33  5493.3   146.4
  5493.3 5788.71  147.45
Permanent Ineff=
       F       F       F       F
#Block Obstruct= 1 ,-1
       0  594.97  146.96
Bank Sta=4282.62,4602.35
XS Rating Curve= 0 ,0
Exp/Cntr=0.3,0.1

Type RM Length L Ch R = 1 ,94049.88,274.6,309.58,299.42
BEGIN DESCRIPTION:
Updated (March 2016)
END DESCRIPTION:
Node Name=AC
XS GIS Cut Line= 6
3006358.8375287813896319.15011663005827.2910196913892288.1234018
3005763.9922617813892178.24599683005763.9922617813891726.4388296
3005778.5801591113891524.29258043005896.2515116913891016.4205646
#Sta/Elev= 30
       0  147.82   199.8   145.7   299.7  147.32 1173.82  145.75 1195.62     148
  1398.6  145.64 1643.36  145.52 1686.45   147.6 1738.26  145.76 1949.66  145.74
  2163.5  145.17 2472.52  145.61    2550   147.7    3375   147.7    3475  144.75
 3825.97  144.22 3905.77  133.44 4073.05   132.9 4109.38  129.83 4131.63  132.86
 4175.97  133.77 4223.52  142.17 4251.96  144.48    4298  144.65    4309     148
    4750   148.4 4802.69  144.94 4957.48  145.14  4971.3  147.29 5368.49  146.73
#Mann= 6 ,-1 , 0
       0     .07       0 1949.66     .12       0  2163.5     .07       0
 3825.97     .04       0 4251.96     .07       0 4957.48     .15       0
#XS Ineff= 4 ,-1
       0 1983.02  146.96                            4298  4971.3   146.2
  4971.3 5368.49  147.29
Permanent Ineff=
       F       F       F       F
#Block Obstruct= 3 ,-1
       0  239.76  146.86                          4971.3 5368.49  146.84
Bank Sta=3825.97,4251.96
XS Rating Curve= 0 ,0
Exp/Cntr=0.3,0.1

Type RM Length L Ch R = 1 ,93740.3 ,854.24,1015.49,680.15
BEGIN DESCRIPTION:
Updated (March 2016)
END DESCRIPTION:
XS GIS Cut Line= 6
  3007022.957263 13895359.787534 3006444.543722213892444.9019596
 3006109.170049113892100.2418878  3006064.81154213892054.6553648
 3006061.349934813892025.1400038 3005932.359707213890926.8039459
#Sta/Elev= 30
       0   145.7  244.73  145.01  264.71   146.4  329.64  144.65  419.54  145.64
  689.24  144.18  884.02  145.99     904  144.19  948.95  146.54 1013.88  144.97
 2676.62  144.77 2725.89  141.97 2764.94  135.34 3329.04   132.7 3342.24  128.34
 3356.09  128.93 3370.72  134.38 3455.61  140.97 3473.49  144.38 3479.57  143.52
 3483.75  144.66  3495.6  147.89 3525.75   142.2 3545.75   142.6  3555.9  144.95
 3949.43  144.82 3979.32   147.8 4203.48  144.41  4278.2  145.78 4651.81  146.58
#Mann= 4 ,-1 , 0
       0     .07       0 2676.62     .04       0  3495.6     .07       0
  3555.9     .07       0
#XS Ineff= 5 ,-1
       0 1034.76  147.46 2676.62    3172     144 3583.94 3857.26     146
 3857.26 4534.73  146.58    3444    3556     144
Permanent Ineff=
       F       T       F       F       T
#Block Obstruct= 2 ,-1
                         4036.59    4479     146
Bank Sta=2676.62,3483.75
XS Rating Curve= 0 ,0
Exp/Cntr=0.5,0.3

Type RM Length L Ch R = 2 ,93317   ,,,
BEGIN DESCRIPTION:
Pipeline Easement Crossing
END DESCRIPTION:
Node Name=TN PIPELINE ESMT
Bridge Culvert--1,0,-1,-1, 0
Deck Dist Width WeirC Skew NumUp NumDn MinLoCord MaxHiCord MaxSubmerge Is_Ogee
30,259,2.6,0, 6, 6, 138, , 0.98, 0, 4,4,,
    2600    3172    3232    3242    3302    3600
     144     144     138     138     144     144
                                                
    2882    3150    3210    3220    3280    3600
     144     144     138     138     144     144
                                                
BR Coef=-1 , 0 , 0 ,, 0 ,,,0.8,-1,,0,
WSPro=,,,, 1 ,,,, 0 ,,,, 0 ,,,,-1 ,-1 ,-1 , 0 , 0 , 0 , 0 , 0
Culvert=2,5,10,310,0.013,0.5,1,8,1,128.84,3326.5,128.78,3376.5,Culvert #4  , 0 ,20
Culvert Bottom n=0.013
Culvert=2,5,10,310,0.013,0.5,1,8,1,128.86,3339.5,128.79,3389.5,Culvert #2  , 0 ,20
Culvert Bottom n=0.013
Culvert=2,4,6,310,0.013,0.5,1,8,1,130.89,3353.5,130.64,3403.5,Culvert #1  , 0 ,20
Culvert Bottom n=0.013
Culvert=2,4,6,310,0.013,0.5,1,8,1,130.78,3361.5,130.65,3411.5,Culvert #3  , 0 ,20
Culvert Bottom n=0.013
BC Design=,, 0 ,, 0 ,,,,,,
BC Use User HTab Curves=0
BC User HTab FreeFlow(D)= 0

Type RM Length L Ch R = 1 ,92724.82,559.57,511.77,496.93
BEGIN DESCRIPTION:
UPDATED (February 2017)
END DESCRIPTION:
XS GIS Cut Line= 5
3007719.2491780213894953.07345243006844.8299951113891942.2901039
 3006722.990015713891810.68997343005987.0689153713890855.7276445
3005790.9180609413890709.9241304
#Sta/Elev= 30
       0   144.4  539.17  144.41  554.15  146.03  599.08   144.2  634.03  145.73
  710.54  144.64  838.71  144.43  853.69  145.94  873.66  143.77 1265.63  143.55
 2441.39  143.76  3135.2  143.28 3140.18  143.32 3234.84  131.92 3309.56  130.74
 3329.32  128.07 3378.59  132.54 3461.75  132.89 3495.91  137.37 3593.54     145
 3653.32  145.97 3762.93  143.87 3892.45  146.62 4355.77  143.87 4519.47  146.59
 4575.04  142.23  4634.9  145.64 4698.18  142.95 4729.66  147.39 4764.58  147.35
#Mann= 8 ,-1 , 0
       0     .07       0  710.54     .12       0 1265.63     .07       0
 2441.39     .07       0  3135.2     .04       0 3593.54     .15       0
 4519.47     .07       0 4698.18     .15       0
#XS Ineff= 2 ,-1
    2880    3150     144 3653.32 4764.58   145.1
Permanent Ineff=
       F       F
#Block Obstruct= 2 , 0
       0                 4565.07       0  144.31
Bank Sta=3140.18,3593.54
XS Rating Curve= 0 ,0
Exp/Cntr=0.3,0.1

Type RM Length L Ch R = 1 ,92213.05,385.4,785.94,950.63
BEGIN DESCRIPTION:
UPDATED (February 2017)
END DESCRIPTION:
Node Name=AB
XS GIS Cut Line= 5
 3007876.631409213894882.57917093007487.91991627 13891968.569907
3007147.3799149413891551.40998023007033.6987118613891391.2229646
3006122.9803889413890342.5095108
#Sta/Elev= 30
       0  144.51 1344.07  144.04 1469.04  143.39 2286.56  141.93 2669.83  141.23
 2719.83  143.44 2854.82  140.52 3014.46  144.09 3223.45  140.44 3377.89  143.71
 3382.67  143.78 3478.32   131.3 3590.23  127.83 3679.74   132.3 3714.72  138.23
 3804.64  143.97 3983.75  143.51 4149.37  144.79 4344.23  141.34 4414.17  135.68
 4469.13  135.58  4519.1  142.23 4569.06  145.09 4683.97  143.59 4833.86  145.93
 4893.81     142 4953.77   145.6 5013.72  142.32 5052.09  147.38 5063.68  147.82
#Mann= 8 ,-1 , 0
       0     .07       0 1344.07     .12       0 1469.04     .07       0
 2286.56     .07       0 3377.89     .04       0 3804.64     .15       0
 3983.75     .07       0 5052.09     .15       0
#XS Ineff= 2 ,-1
 2316.69 3348.68  143.12 4658.99 5063.68  144.77
Permanent Ineff=
       F       F
#Block Obstruct= 2 ,-1
 4149.37 4559.07  144.79 4883.82 5063.68   143.6
Bank Sta=3382.67,3804.64
XS Rating Curve= 0 ,0
Exp/Cntr=0.3,0.1

Type RM Length L Ch R = 1 ,91427.11,471.39,483.13,469.42
BEGIN DESCRIPTION:
UPDATED (February 2017)
END DESCRIPTION:
XS GIS Cut Line= 5
3008163.3526205313894966.42086673007737.91777585 13891657.479978
3007717.01000927  13891204.669863007677.95004803 13890761.969958
3007456.2060689513888986.6798734
#Sta/Elev= 30
       0  144.15  604.31  145.27 1338.46  142.22  2315.3  141.97 2347.31  144.06
 2891.68  143.85 3091.45   142.6  3136.4  140.54 3171.35  142.33 3336.16  142.95
 3469.98  140.24 3630.77  143.67  3640.7  143.66 3734.91  132.67 3968.37  130.02
 4007.71  126.47 4047.04  131.96 4169.96  133.41 4243.87  142.56 4258.86  142.24
 4303.84  132.34 4673.65  132.09 5103.43  143.35 5238.36  141.97 5708.12  143.89
  5758.1  143.62 5808.07  140.57 5898.03  144.15    5963  140.47 6022.96  145.14
#Mann= 4 ,-1 , 0
       0     .07       0  2315.3     .07       0 3630.77     .04       0
 4243.87     .07       0
#XS Ineff= 2 ,-1
 2354.21 3632.71  143.66 5198.38 6022.96   143.2
Permanent Ineff=
       F       F
#Block Obstruct= 2 ,-1
 4243.87 5023.47  142.24 5793.08 6022.96  142.32
Bank Sta=3640.7,4243.87
XS Rating Curve= 0 ,0
Exp/Cntr=0.3,0.1

Type RM Length L Ch R = 1 ,90943.98,397.97,474.62,519.56
BEGIN DESCRIPTION:
UPDATED (February 2017)
END DESCRIPTION:
XS GIS Cut Line= 4
3008347.9677368613895020.4050107 3008189.805979713891095.9312323
3008114.11879511  13890632.348173007968.3241391913888222.2076491
#Sta/Elev= 30
       0  143.64 2199.42  142.36  2424.2  140.59  2449.2  142.74 2699.12  142.59
 2789.09  140.14 3163.97  143.73 3343.91   142.4  3373.9  139.89 3473.87  143.22
  3688.8  140.49 3839.75  143.95 3844.63  143.98 3937.56  131.56 4110.71  129.48
 4150.29  126.24 4179.88  130.81 4239.01  131.68 4293.22  139.65  4352.4     142
 4672.32   144.6 5152.25  141.86 5227.24  144.02 5852.14  142.33 5947.12  144.28
 5992.11  143.91 6012.11  140.56 6497.03  139.53 6607.02  142.86 6811.98   142.7
#Mann= 4 ,-1 , 0
       0     .07       0 2199.42     .07       0 3839.75     .04       0
  4352.4     .07       0
#XS Ineff= 2 ,-1
 2258.35 3832.78  143.53 4492.35 6811.98  143.26
Permanent Ineff=
       F       F
#Block Obstruct= 2 , 0
       0  144.91  145.03 5947.12       0   142.5
Bank Sta=3844.63,4352.4
XS Rating Curve= 0 ,0
Exp/Cntr=0.3,0.1

Type RM Length L Ch R = 1 ,90469.36,706,713.14,720.38
BEGIN DESCRIPTION:
UPDATED (February 2017)
END DESCRIPTION:
XS GIS Cut Line= 5
 3008532.582853213895074.38915473008622.6099041113891008.9199234
3008622.60990411 13890862.7099143008617.3002034413890650.3543676
 3008508.8388062 13888150.357071
#Sta/Elev= 30
       0  143.45 2053.49  142.37 2103.35  144.23  2288.2  140.56 2453.07  143.85
 2632.92  140.05 2797.79  143.79 2962.66  140.67 3132.52  143.83 3357.34   140.4
 3842.09  143.91 3862.05  143.82    3877  139.45  3946.8  132.38 4178.54  129.37
 4207.78  125.96 4236.34  129.72 4279.31  130.12 4375.68  141.66 4445.06  144.02
 4754.73  141.92 5044.41  144.55 5129.32  142.23 5174.27  144.85 5793.61  141.94
  5988.4  145.07 6038.35  144.22 6053.33  139.99 6898.05  140.28 6927.39  141.34
#Mann= 5 ,-1 , 0
       0     .07       0 2053.49     .07       0 3842.09     .04       0
 4375.68     .07       0 6898.05     .12       0
#XS Ineff= 2 ,-1
 2111.99  3859.5  143.78 4609.88 6927.39  142.89
Permanent Ineff=
       F       T
#Block Obstruct= 2 , 0
       0                  5988.4       0   142.5
Bank Sta=3862.05,4375.68
XS Rating Curve= 0 ,0
Exp/Cntr=0.3,0.1

Type RM Length L Ch R = 1 ,89756.23,175.18,156.89,155.73
BEGIN DESCRIPTION:
UPDATED (February 2017)
END DESCRIPTION:
XS GIS Cut Line= 6
3009170.0700952713895260.79987113009330.7600626113891177.1499019
3009320.1199920313890989.10008123009309.0701453513890781.0299593
3009255.7628372813888019.95641323009254.4567375313887952.3112073
#Sta/Elev= 30
       0  143.03 2007.15  142.75 2577.99  140.99 2907.74  144.35 3067.62  140.98
 3297.44  143.72 3562.23  140.51 3752.09  143.73 3926.95  140.71 4152.23  144.02
 4221.11   136.9 4245.69  130.24 4328.38  129.09  4357.4  125.12 4386.42  129.72
 4425.24  129.66 4449.54  135.46  4513.5  141.99 4908.01   143.6 4967.94  140.08
 5022.87   131.8 5087.79  131.75 5172.69  132.03 5257.58  142.94 5392.42  143.73
 6970.47  140.59 7060.36  144.36 7175.22  138.64 7292.81  140.11 7312.79  140.42
#Mann= 5 ,-1 , 0
       0     .07       0 2007.15     .07       0 4152.23     .04       0
  4513.5     .07       0 7292.81     .12       0
#XS Ineff= 1 ,-1
 2047.43 4148.78  143.99
Permanent Ineff=
       F
#Block Obstruct= 2 ,-1
 4908.01 5257.58  142.94  7110.3 7312.79   142.5
Bank Sta=4152.23,4513.5
XS Rating Curve= 0 ,0
Exp/Cntr=0.3,0.1
