HEC-RAS study U100-00-00.prj: U100-00-00

--- U100-00-00.g01 (geometry) --- (continued)

Type RM Length L Ch R = 1 ,72607.04,570.32,575.35,579.02
XS GIS Cut Line= 5
3019413.4980991913880636.28450083019377.2094578613880573.2724877
3018889.9601042713880140.85996673018729.3600317813879983.6900054
3018295.0899029413879630.1001614
#Sta/Elev= 30
       0  125.72   47.62  125.39   67.87  124.43  122.44  124.03  251.74  124.47
   460.6  122.65  624.71  122.81  714.22  124.21  754.13  122.27  759.61  122.08
  794.41  112.32   804.4  111.47  808.57  108.36  820.24  107.94  821.44   108.3
   824.7   111.6  839.85  113.08  873.98  123.82  878.97  124.47  893.95  123.84
  940.22  125.68 1077.73  123.63 1142.16  123.58 1157.03   122.9 1236.32  122.27
 1345.35  125.26 1360.22  124.82 1375.09  125.67 1409.78  126.08  1508.9  126.16
#Mann= 5 ,-1 , 0
       0     .15       0   47.62     .07       0  754.13     .04       0
  878.97     .07       0  940.22     .15       0
#XS Ineff= 2 ,-1
       0  500.39  124.48 1062.87  1508.9  124.12
Permanent Ineff=
       F       F
Bank Sta=754.13,878.97
XS Rating Curve= 0 ,0
Exp/Cntr=0.3,0.1

Type RM Length L Ch R = 1 ,72031.7 ,94.52,93.9,93.21
XS GIS Cut Line= 4
3019413.3202780313880626.83241993019386.0503194513880576.7249086
3019411.3393108513879878.3053737 3018885.061820113879267.3705719
#Sta/Elev= 30
       0  125.75   37.91  125.59   57.05  124.43  126.94  124.76  166.87  123.85
  191.83  124.44  226.77  123.38  296.66  124.13  356.57  122.92  386.52  123.74
   586.2  123.74  706.01  121.43  820.63  121.77  865.43  122.78  920.18  122.25
  926.84  121.82  973.34  105.17  987.69  104.47 1039.64   122.5 1044.62   123.1
 1059.55  122.28 1069.51  123.25  1111.4  123.71 1233.77  121.94 1283.54   124.4
 1368.16  124.67 1472.69  123.94 1527.44  122.98  1537.4  122.06 1562.28  122.52
#Mann= 5 ,-1 , 0
       0     .15       0   37.91     .07       0  920.18     .04       0
 1044.62     .07       0  1111.4     .15       0
#XS Ineff= 2 ,-1
       0  777.27   123.8  1114.3 1562.28   123.8
Permanent Ineff=
       F       F
#Block Obstruct= 2 , 0
       0                 1472.69       0  123.94
Bank Sta=920.18,1044.62
XS Rating Curve= 0 ,0
Exp/Cntr=0.3,0.1

Type RM Length L Ch R = 1 ,71937.8 ,85.25,87.92,92.4
XS GIS Cut Line= 4
3019413.1211314513880616.23270363019394.8915091213880580.1770014
3019425.0236666913879747.99067373018995.7256407713879261.3066077
#Sta/Elev= 30
       0  125.79   27.17  125.52   50.37  124.53  125.17  124.62  155.09  123.74
  189.99   124.3  214.93  123.35  279.75  124.13  344.57  123.07  494.17  124.06
  608.85  122.41  618.83  123.12  673.68  121.56  948.01  122.14  952.14  121.86
  974.65  113.22 1004.25  104.52 1009.25  104.43 1015.58  104.69 1066.73  122.14
 1072.82  122.69 1133.99  123.41 1162.67     124 1217.58  123.38 1292.46  121.37
 1337.39  123.48 1432.24  123.85 1492.15  122.75 1507.12  121.53  1522.1  121.88
#Mann= 5 ,-1 , 0
       0     .15       0   27.17     .07       0  948.01     .04       0
 1072.82     .07       0 1133.99     .15       0
#XS Ineff= 2 ,-1
       0  860.18  123.86 1162.67  1522.1     124
Permanent Ineff=
       F       F
#Block Obstruct= 2 , 0
       0                 1382.32       0  123.99
Bank Sta=948.01,1072.82
XS Rating Curve= 0 ,0
Exp/Cntr=0.3,0.1

Type RM Length L Ch R = 1 ,71849.88,5.36,71.2,131.32
Node Name=R
XS GIS Cut Line= 4
3019413.1381917713880607.64184153019412.5732322813880587.0815152
3019446.6177836113879646.84881563019142.7725907713879255.2429715
#Sta/Elev= 30
       0  125.54   18.87  125.33   95.24  124.13  115.15  124.51     150  123.58
  159.95  124.42  179.87  124.55  204.76  123.51  329.21  123.03  483.53  124.06
  568.15   122.7  583.09  123.51  593.04  122.53  722.47  121.38   737.4  121.99
  802.12  121.46  916.61   122.5  964.59  122.09  966.25  122.59  1031.3  104.69
 1038.57  104.11 1043.29  104.61 1072.59   114.5 1093.34  122.69 1095.24  122.87
 1105.16  122.28    1149  123.06 1313.33  123.07 1407.51  120.76 1457.08  121.22
#Mann= 5 ,-1 , 0
       0     .15       0   18.87     .07       0  966.25     .04       0
 1095.24     .07       0    1149     .15       0
#XS Ineff= 2 ,-1
       0  924.59  123.86 1224.12 1457.08  122.76
Permanent Ineff=
       F       F
#Block Obstruct= 2 , 0
       0                 1352.99       0  122.24
Bank Sta=966.25,1095.24
XS Rating Curve= 0 ,0
Exp/Cntr=0.5,0.3

Type RM Length L Ch R = 1 ,71778.68,17.96,20.35,53.55
BEGIN DESCRIPTION:
Upstream Section - 12" PIPELINE
END DESCRIPTION:
XS GIS Cut Line= 3
3019414.5870077813880601.93680043019416.3238809413880553.9683924
 3019463.3641412 13879254.819744
#Sta/Elev= 30
       0  125.45  10.906  125.23  69.345  124.15  85.105  124.52 112.686  123.71
 136.326  124.44 148.146   124.3 156.026  123.55 179.666  123.82 254.527  123.05
 282.108  123.61 376.669  123.84  435.77  122.74  455.47  123.55  471.23  122.39
 561.852  121.29 577.612  121.93 613.072  121.37 719.454   122.5 757.144  122.09
 762.566  122.51 806.584  111.54 843.952  104.02 847.608  103.66 851.942  103.99
 903.722  120.79 924.337  122.541015.998  122.571050.418  122.391062.239   123.1
#Mann= 5 ,-1 , 0
       0     .15       0  10.906     .07       0 762.566     .04       0
 924.337     .07       01015.998     .15       0
#XS Ineff= 2 ,-1
       0  762.57  123.86  924.341062.239  122.76
Permanent Ineff=
       F       F
Bank Sta=762.566,924.337
XS Rating Curve= 0 ,0
Skew Angle= 38
Exp/Cntr=0.5,0.3

Type RM Length L Ch R = 3 ,71768.64,,,
BEGIN DESCRIPTION:
12" PIPELINE
U00_800
END DESCRIPTION:
Node Name=12" PIPELINE
Bridge Culvert--1,0,-1,-1, 0
Deck Dist Width WeirC Skew NumUp NumDn MinLoCord MaxHiCord MaxSubmerge Is_Ogee
9,1,2.6,38, 7, 7, , , 0.98, 0, 0,0,,
 747.034 775.505 802.534 836.024 869.515 902.769 927.828
  121.64  121.64  121.63  121.62  121.62  121.61   121.6
  120.64  120.64  120.63  120.62  120.62  120.61  120.61
 747.034 775.505 802.534 836.024 869.515 902.769 927.828
  121.64  121.64  121.63  121.62  121.62  121.61   121.6
  120.64  120.64  120.63  120.62  120.62  120.61  120.61
Pier Skew, UpSta & Num, DnSta & Num=  ,802.534, 2 ,802.534, 2 , 0 , 0 , 0 ,,
     1.4     1.4
     100   121.3
     1.4     1.4
     100   121.3
Pier Skew, UpSta & Num, DnSta & Num=  ,836.024, 2 ,836.024, 2 , 0 , 0 , 0 ,,
     1.4     1.4
     100   121.3
     1.4     1.4
     100   121.3
Pier Skew, UpSta & Num, DnSta & Num=  ,869.515, 2 ,869.515, 2 , 0 , 0 , 0 ,,
     1.4     1.4
     100   121.3
     1.4     1.4
     100   121.3
Pier Skew, UpSta & Num, DnSta & Num=  ,901.981, 2 ,902.769, 2 , 0 , 0 , 0 ,,
     1.4     1.4
     100   121.3
     1.4     1.4
     100   121.3
BR Coef=-1 , 1 , 1 ,0.9, 0 ,,,0.8,-1,1.2,0,
WSPro=,,,, 1 ,,,, 0 ,,,, 0 ,,,,-1 ,-1 ,-1 , 0 , 0 , 0 , 0 , 0
BC Design=,, 0 ,, 0 ,,,,,,
BC Use User HTab Curves=0
BC User HTab FreeFlow(D)= 0

Type RM Length L Ch R = 1 ,71758.34,1.52,1.84,1.55
BEGIN DESCRIPTION:
Downstream Section - 12" PIPELINE
END DESCRIPTION:
XS GIS Cut Line= 3
3019431.15062295 13880589.2265243019432.88749611 13880541.258116
3019479.9277563513879242.1094676
#Sta/Elev= 30
       0  125.24   4.381  125.18  61.465  124.09  85.105  124.51 100.865  123.76
 128.446  124.52 140.266  124.33 152.086  123.39 262.408   122.8 349.089  123.66
 396.369   123.5  443.65  122.36 561.852  121.74 569.732  121.26 652.473  121.07
 715.514  122.41 747.034  122.65 752.716  122.26 796.104  111.54 831.651  104.99
 833.471  104.02 837.127  103.66 841.461  103.99 882.383  117.19  932.69  122.32
 936.157  122.72 991.318  122.411018.898  123.121026.778   122.51062.239  122.53
#Mann= 4 ,-1 , 0
       0     .15       0   4.381     .07       0 752.716     .04       0
  932.69     .07       0
#XS Ineff= 2 ,-1
       0  747.03  123.86  936.161062.239  122.76
Permanent Ineff=
       F       F
Bank Sta=752.716,932.69
XS Rating Curve= 0 ,0
Skew Angle= 38
Exp/Cntr=0.5,0.3

Type RM Length L Ch R = 1 ,71756.49,135.69,137.93,127.2
BEGIN DESCRIPTION:
Upstream Section - BARKER CYPRESS RD
END DESCRIPTION:
XS GIS Cut Line= 3
3019432.6434021113880588.08118513019434.3802752813880540.1127771
3019481.4205355213879240.9641287
#Sta/Elev= 30
       0  125.21    3.79  125.08  18.912  124.54  61.465  124.06  85.105  124.53
 100.865  123.73 112.686  124.45 124.506  124.53 140.266  124.26 148.146  123.53
 238.767  123.13 270.288  122.65 337.269  123.62 392.429  123.53  443.65  122.33
 636.713  121.08 672.173  121.35 711.574  122.38 747.034  122.66 752.117  122.23
 795.158  111.54 830.705  104.99 832.526  104.02 932.185  122.22 932.217  122.23
 940.097  122.79 979.497  122.251018.898  122.961042.538  122.371062.239   122.6
#Mann= 4 ,-1 , 0
       0     .15       0    3.79     .07       0 752.117     .04       0
 932.185     .07       0
#XS Ineff= 2 ,-1
       0 766.734  123.86 919.9711062.239  122.76
Permanent Ineff=
       F       F
Bank Sta=752.117,932.217
XS Rating Curve= 0 ,0
Skew Angle= 38
Exp/Cntr=0.5,0.3

Type RM Length L Ch R = 3 ,71687.63,,,
BEGIN DESCRIPTION:
BARKER CYPRESS RD
U00_800
END DESCRIPTION:
Node Name=BARKER CYPRESS
Bridge Culvert--1,0,-1,-1, 0
Deck Dist Width WeirC Skew NumUp NumDn MinLoCord MaxHiCord MaxSubmerge Is_Ogee
11.5,92,2.6,38, 60, 60, , , 0.98, 0, 0,0,,
       0  22.695  37.825  61.465  69.345  77.225 120.566 128.446 148.146 156.026
 163.906 187.547 195.427 199.367 207.247 211.187 219.067 226.947 234.827 238.767
 246.647 254.527 289.988 321.508 349.089 372.729 380.609 388.489  416.07  431.83
  443.65  451.53 518.511 522.451 530.331 534.271 550.031 565.792 585.492 593.372
 597.312 691.873 695.814 750.974 754.914 762.794 766.734 798.255 829.775 865.236
 928.277 932.217 936.157 940.097 944.037 971.617 975.557 987.3781026.7781062.239
  126.14  126.01  126.12  125.95  125.81  125.18  125.11  124.94  124.91  124.73
  124.82  124.55  124.77  124.63  124.83  124.63  124.85  124.64  124.72  124.56
   124.7  124.43  124.44  124.12  124.27     124  123.98  124.16  123.86  124.09
  123.89  124.02  124.12  124.25  124.13  124.33  124.52  124.42  124.61  124.57
  124.26   124.2  125.19   125.2  127.29  127.29  127.29  127.29  127.28  127.28
  127.27  127.27  127.27  127.27  125.89  125.89  123.92  123.99  123.12  122.76
       0       0       0       0       0       0       0       0       0       0
       0       0       0       0       0       0       0       0       0       0
       0       0       0       0       0       0       0       0       0       0
       0       0       0       0       0       0       0       0       0       0
       0       0       0       0       0       0  119.94  119.66  119.93     120
  119.99  111.81       0       0       0       0       0       0       0       0
       0  57.525  69.345  77.225 120.566 128.446 136.326 144.206 148.146 156.026
 163.906 187.547 191.487 195.427 199.367 207.247 211.187 219.067 226.947 234.827
 238.767 246.647 254.527 289.988 297.868 309.688 321.508 349.089 372.729 380.609
 388.489 400.309  408.19  416.07  431.83  443.65  451.53 490.931 510.631 518.511
 526.391 640.653 652.473 687.933 691.873 719.454 723.394 727.334 731.274 861.296
 892.816 896.756 904.636 908.576 944.037 983.4371018.8981046.4781058.2981062.239
  126.14  125.99  125.81  125.18  125.11  124.94  124.97  124.82  124.91  124.73
  124.82  124.55  124.58  124.77  124.63  124.83  124.63  124.85  124.64  124.72
  124.56   124.7  124.43  124.44  124.28  124.33  124.12  124.27     124  123.98
  124.16     124  124.03  123.86  124.09  123.89  124.02     124   124.2  124.12
  124.26  124.21  124.91  125.04   125.8   125.8  127.08  127.13  127.15  127.14
  127.14  127.16  127.22  125.39  124.87  122.83  122.61  122.58  122.58  122.76
       0       0       0       0       0       0       0       0       0       0
       0       0       0       0       0       0       0       0       0       0
       0       0       0       0       0       0       0       0       0       0
       0       0       0       0       0       0       0       0       0       0
       0       0       0       0       0       0       0       0  119.94  120.05
  120.04       0       0       0       0       0       0       0       0       0
Pier Skew, UpSta & Num, DnSta & Num=  ,796.127, 2 ,763.661, 2 , 0 , 0 , 0 ,,
     1.2     1.2
     100     122
     1.2     1.2
     100     122
Pier Skew, UpSta & Num, DnSta & Num=  ,830.012, 2 ,797.309, 2 , 0 , 0 , 0 ,,
     1.2     1.2
     100     122
     1.2     1.2
     100     122
Pier Skew, UpSta & Num, DnSta & Num=  ,864.29, 2 ,830.642, 2 , 0 , 0 , 0 ,,
     1.2     1.2
     100     122
     1.2     1.2
     100     122
Pier Skew, UpSta & Num, DnSta & Num=  ,897.702, 2 ,861.296, 2 , 0 , 0 , 0 ,,
     1.2     1.2
     100     122
     1.2     1.2
     100     122
BR Coef=-1 , 1 , 1 ,1.25, 0 ,,,0.8,-1,2,0,
WSPro=,,,, 1 ,,,, 0 ,,,, 0 ,,,,-1 ,-1 ,-1 , 0 , 0 , 0 , 0 , 0
BC Design=,, 0 ,, 0 ,,,,,,
BC Use User HTab Curves=0
BC User HTab FreeFlow(D)= 0

Type RM Length L Ch R = 1 ,71618.56,95.68,37.58,4.34
BEGIN DESCRIPTION:
Downstream Section - BARKER CYPRESS RD
END DESCRIPTION:
XS GIS Cut Line= 3
3019544.3859607713880502.33627793019546.1228339413880454.3678699
3019593.1630941913879155.2192214
#Sta/Elev= 30
       0  124.41  26.477  125.62  41.765   124.2  73.285  124.91  92.985   124.4
 144.206  124.58 159.966  123.85 226.947   124.9 274.228  124.11 293.928     123
 309.688  121.05 329.389  121.34 337.269  122.25 345.149  124.14 376.669  125.01
 514.571  123.17 542.151  123.56 624.893  122.31 636.713  122.78 714.505  122.18
 743.094  121.19 813.708  107.94 821.533  104.43  827.86  102.93 832.297  104.63
 882.919  115.06 907.796  121.54 916.457  122.43 944.037  120.971062.239  121.24
#Mann= 4 ,-1 , 0
       0     .15       0 714.505     .07       0 743.094     .04       0
 907.796     .07       0
#XS Ineff= 3 ,-1
       0 356.969  124.63 356.969  749.54  122.29 892.8161062.239  121.88
Permanent Ineff=
       F       F       F
#Block Obstruct= 2 , 0
       0  26.477  125.62               0
Bank Sta=743.094,907.796
XS Rating Curve= 0 ,0
Skew Angle= 38
Exp/Cntr=0.5,0.3

Type RM Length L Ch R = 1 ,71580.98,109.77,106.23,83.69
XS GIS Cut Line= 4
 3020213.722548613880475.89472973020100.9904906213880279.0398084
3019589.1181547813879385.19907643019597.55613002 13879152.158532
#Sta/Elev= 30
       0  125.14   59.18  124.38   88.77  122.16  113.42  122.11  152.88  124.43
  291.54  124.66   361.2  123.66  401.01  120.26   465.7  120.49   485.6  119.43
  644.83  123.69  863.78  122.56  913.54  121.24  943.39  118.99 1042.91  122.22
 1081.18  121.64 1097.65  121.54 1118.73  120.48 1174.33  112.04 1187.13  106.99
 1191.48  102.83 1201.15  101.15 1206.91  102.15 1215.07  108.31 1221.95  110.66
 1259.29  115.06 1291.61  121.52 1301.54  122.44  1331.3  121.04 1490.07   121.2
#Mann= 4 ,-1 , 0
       0     .15       0 1081.18     .07       0 1097.65     .04       0
 1301.54     .07       0
#XS Ineff= 3 ,-1
       0  138.08  123.85  138.08 1013.06  121.38 1301.54 1490.07   122.5
Permanent Ineff=
       F       F       F
Bank Sta=1097.65,1301.54
XS Rating Curve= 0 ,0
Exp/Cntr=0.3,0.1

Type RM Length L Ch R = 1 ,71474.76,96.13,97.51,97.03
XS GIS Cut Line= 5
3020260.2788859513880477.19984523020158.1780402813880237.3430414
3019945.5259065313879737.77875193019632.3273859513879270.4906444
3019636.6738339413879150.4534829
#Sta/Elev= 30
       0  125.08   49.19  124.84  108.21  121.97  157.39  124.67  295.55  124.29
  350.34  122.63  380.23  120.27  544.61  123.76  564.53  122.87  614.34  123.59
  619.32  122.28  659.17  120.08  684.08  119.83  723.93  122.61  848.43  122.55
  977.86  119.29  1037.6  122.51 1113.21  121.76 1142.14  120.87 1159.87  119.62
 1181.44  114.71 1202.67  112.45 1212.76  107.74 1220.44  101.48 1224.97  101.15
 1229.81  101.86 1233.69  104.89 1243.66  108.24  1311.4  120.83 1486.28  121.85
#Mann= 4 ,-1 , 0
       0     .15       0 1113.21     .07       0 1142.14     .04       0
  1311.4     .07       0
#XS Ineff= 2 ,-1
       0   132.8  123.73   132.8 1022.67  121.33
Permanent Ineff=
       F       F
Bank Sta=1142.14,1311.4
XS Rating Curve= 0 ,0
Exp/Cntr=0.3,0.1

Type RM Length L Ch R = 1 ,71377.24,345.25,354.84,352.69
XS GIS Cut Line= 4
3020298.9776274413880478.28514493020202.0588580213880193.4622237
3020036.6625352813879707.3998756 3019672.115692213879153.8288043
#Sta/Elev= 30
       0  125.29   44.39  124.57   83.85  122.09   138.1  124.37  271.27  124.28
  335.75     123  365.66  120.74   385.6  120.57  415.51  122.03  540.13   124.3
  609.92  122.77   649.8  120.49  674.72  120.58  729.55  122.94  928.92  121.46
 1008.65  119.57 1033.57  119.75 1073.44   121.6  1143.9  121.21 1173.11  120.51
 1186.54  119.52 1249.31  109.84 1256.92  107.32 1261.52  102.12 1266.96  100.82
 1272.07  102.09 1279.21  108.08 1340.41   119.8 1357.51  120.51 1477.12  121.55
#Mann= 4 ,-1 , 0
       0     .15       0  1143.9     .07       0 1173.11     .04       0
 1357.51     .07       0
#XS Ineff= 2 ,-1
       0   123.3  123.72   123.3 1078.43  121.65
Permanent Ineff=
       F       F
Bank Sta=1173.11,1357.51
XS Rating Curve= 0 ,0
Exp/Cntr=0.3,0.1

Type RM Length L Ch R = 1 ,71022.41,383.27,446.68,435.03
XS GIS Cut Line= 5
3020431.4537404513880278.39545283020407.9603491113880195.1498844
3020137.0999984413879235.40016343020050.65988261  13879088.70984
3019781.9786614513878993.3865398
#Sta/Elev= 30
       0   124.9    86.5  124.03  146.33  121.06  171.26  121.17  206.17  123.36
  325.83  124.47   445.5  121.14  475.42  122.47  545.23  122.99  615.03  121.53
  724.73  122.49  819.47  121.95  834.43  120.98  884.29  121.06  924.18  118.99
  993.99  120.57 1056.52  120.69 1104.47  119.35 1105.77  120.56 1130.79   113.8
 1142.19  112.51 1157.74   108.8 1164.97  102.23 1170.34  102.06 1176.09  103.46
  1180.8  109.34  1212.9   108.6 1251.99  119.29 1263.83   120.3 1539.09  122.13
#Mann= 4 ,-1 , 0
       0     .15       0 1056.52     .07       0 1105.77     .04       0
 1263.83     .07       0
#XS Ineff= 2 ,-1
       0   231.1  123.62   231.1 1003.96  120.65
Permanent Ineff=
       F       F
Bank Sta=1105.77,1263.83
XS Rating Curve= 0 ,0
Exp/Cntr=0.3,0.1

Type RM Length L Ch R = 1 ,70575.73,369.02,375.02,374.54
BEGIN DESCRIPTION:
Confluence with Dinner Creek (U120-00-00)
END DESCRIPTION:
XS GIS Cut Line= 4
3020535.70648469 13879988.9757563020543.0407876113879317.8639093
3020345.0077191113878555.06983123020161.5687815213877848.4895514
#Sta/Elev= 30
       0  124.71   74.57  123.78  109.37  120.71  164.06  123.02  223.72  123.27
  636.35  121.79   775.9  118.48   815.8  120.73  875.65  121.05  930.52  118.89
   940.5  117.49  965.44  109.55   980.4  107.28  999.65  100.67 1004.61  100.39
 1010.78   101.7 1025.29  109.07 1050.23  109.47 1095.12   121.8 1118.96  120.96
    1145  123.32 1219.82  122.59 1299.62  119.61 1344.51  122.07 1434.29  123.34
 1543.66  122.34 1583.38   119.5 1667.81  123.05 1772.09  124.18 2189.24  125.38
#Mann= 5 ,-1 , 0
       0     .15       0  875.65     .07       0  930.52     .04       0
 1095.12     .07       0 1118.96     .15       0
#XS Ineff= 3 ,-1
       0  183.95  123.13  183.95  860.69  121.04 1234.78 2189.24  121.51
Permanent Ineff=
       F       F       F
Bank Sta=930.52,1095.12
XS Rating Curve= 0 ,0
Exp/Cntr=0.3,0.1

Type RM Length L Ch R = 1 ,70200.7 ,722.22,740.28,736.14
XS GIS Cut Line= 5
3020809.7357922813879604.66484493020830.7101597813878962.0499884
3020786.3001436113878760.45984043020615.12364869 13878384.475028
3020372.0099616913877850.4816734
#Sta/Elev= 30
       0  123.59  164.48  122.05  214.32  122.95  259.18  121.47  398.73  121.03
  468.51  118.05  613.05  120.68  647.87  119.05  652.49  118.65  682.98  109.07
  689.31  108.32  693.97  102.54  696.21   101.4  702.24   99.54  709.11   98.99
  717.57   100.6  721.55  102.65  728.69  108.63  763.55  107.98  801.64  119.83
  810.06  121.31  838.69  120.52   953.9     120  973.81  118.95   998.7  119.19
 1028.56  121.94 1128.11  122.87 1605.58  123.62  1620.5  124.56 1849.23  125.58
#Mann= 5 ,-1 , 0
       0     .15       0  613.05     .07       0  647.87     .04       0
  810.06     .07       0  838.69     .15       0
#XS Ineff= 2 ,-1
       0  578.16  120.51  859.34 1949.23  120.94
Permanent Ineff=
       F       F
Bank Sta=647.87,810.06
XS Rating Curve= 0 ,0
Exp/Cntr=0.3,0.1

Type RM Length L Ch R = 1 ,69460.43,453.32,459.24,467.77
Node Name=Q
XS GIS Cut Line= 5
3021614.0980286913879727.00088633021594.0751028713879485.8255156
 3021538.109991713878811.71990843021459.39066094 13878226.128888
 3021410.214578213877860.3090816
#Sta/Elev= 30
       0  122.58  138.29  122.33  227.19  119.57  570.27  121.21  709.53  118.61
   754.3     121  830.11  120.73   848.8  119.76  868.69  118.12  898.54   108.6
   923.4  105.73  928.36  104.64  935.05  100.34  942.91   99.99  954.11  101.78
  958.15  104.46  963.12  105.91  978.01  107.29 1017.73  120.89 1032.63  121.89
 1051.48  121.47 1067.39  122.65 1112.07  122.61 1191.52  120.05 1345.44  122.31
 1489.43   120.6 1624.02  122.85  1753.7  121.53 1788.62  123.54  1878.4  124.37
#Mann= 5 ,-1 , 0
       0     .15       0  830.11     .07       0   848.8     .04       0
 1032.63     .07       0 1051.48     .15       0
#XS Ineff= 2 ,-1
       0  843.83  120.59 1017.73  1878.4  120.89
Permanent Ineff=
       F       F
Bank Sta=848.8,1032.63
XS Rating Curve= 0 ,0
Exp/Cntr=0.3,0.1

Type RM Length L Ch R = 1 ,69001.19,815.58,821.16,823.78
XS GIS Cut Line= 6
 3022073.473094213879742.28792923022045.6647508613879438.2898495
3021995.8498898613878893.7200725 3021994.300024213878794.4200743
3021992.4401197713878675.04006373021963.1242335313877882.8769498
#Sta/Elev= 30
       0  121.34  152.63  118.44   290.5  120.14  439.49  116.73  504.12  119.73
  568.75  120.25  648.29  119.98  712.91  117.35   767.6  120.65  807.37  120.81
  857.08     120  866.73  118.94  911.11  104.71  926.55   106.7  933.43  100.86
  942.11  100.61  953.42  101.29  959.38  105.74  972.27  105.07 1021.07  120.77
 1031.02  122.09  1069.3  122.19 1150.63  121.81 1195.53  119.67 1405.04   122.5
 1459.91  120.19 1644.35  122.18 1743.97  120.41 1773.86  122.23 1863.52  122.44
#Mann= 5 ,-1 , 0
       0     .15       0  807.37     .07       0  857.08     .04       0
 1031.02     .07       0  1069.3     .15       0
#XS Ineff= 2 ,-1
       0  842.17   120.1  1019.8 1863.52  120.35
Permanent Ineff=
       F       F
#Block Obstruct= 2 , 0
       0   29.54  121.36               0
Bank Sta=857.08,1031.02
XS Rating Curve= 0 ,0
Exp/Cntr=0.3,0.1

Type RM Length L Ch R = 1 ,68180.03,1050.76,1049.08,942.84
XS GIS Cut Line= 6
3022830.3708586113879767.4755429 3022822.081505113879446.2124058
 3022809.059877613878941.55002943022813.5300130213878820.8898376
3022819.3098571213878664.79008423022792.2072210313878023.3638736
#Sta/Elev= 30
       0  121.32   84.05  119.84   93.94   121.2  103.83  119.82  148.32  118.25
  207.65   120.3  296.65  120.46  371.35  119.44  416.34  117.64  556.29  119.75
  636.26  118.72  686.25  116.58  833.99  117.12  855.18  118.61  860.07  118.53
  904.82  105.02  919.22   104.3  930.13  105.06  935.22  100.55  949.92    99.9
  958.53  100.83  963.14  105.51  969.35  106.02  1010.4  118.91 1020.16  120.23
 1052.68  119.81 1207.66  118.66 1312.17  120.99 1466.45  122.26 1745.15  122.86
#Mann= 5 ,-1 , 0
       0     .15       0  833.99     .07       0  855.18     .04       0
 1020.16     .07       0 1052.68     .15       0
#XS Ineff= 3 ,-1
       0  207.65   120.3  207.65  556.29  119.75  556.29  850.35  118.64
Permanent Ineff=
       F       F       F
Bank Sta=855.18,1020.16
XS Rating Curve= 0 ,0
Exp/Cntr=0.3,0.1

Type RM Length L Ch R = 1 ,67130.95,87.58,173.11,202.41
XS GIS Cut Line= 5
3023813.2235516913879800.18282653023866.8700979513878924.4299849
3023779.9099700313878784.53984473023703.5098603713878670.4298367
 3023425.887712213878053.7457026
#Sta/Elev= 30
       0  121.63   69.79  120.92    99.7  118.74  114.66  118.73  154.54  121.56
  483.56  120.93  498.52  121.78  643.09  120.19  687.96  121.04   824.1  119.87
  847.48  117.65  892.37  117.58  917.33     116  947.27  107.54  962.25  106.47
   992.2  106.75 1017.15   102.8 1029.74  102.12 1038.28  100.54 1042.92   98.42
  1049.5  100.65 1050.86  102.21 1056.82  104.69 1076.44  109.36 1105.87  118.75
 1115.68  120.12 1135.29  119.16 1164.72  121.33 1239.11  119.99 1855.73  121.84
#Mann= 4 ,-1 , 0
       0     .15       0   824.1     .07       0  892.37     .04       0
 1115.68     .07       0
#XS Ineff= 2 ,-1
       0  154.54  121.56  154.54  837.54  118.77
Permanent Ineff=
       F       F
#Block Obstruct= 2 , 0
       0                 1840.81       0  122.25
Bank Sta=892.37,1115.68
XS Rating Curve= 0 ,0
Exp/Cntr=0.5,0.3

Type RM Length L Ch R = 1 ,66957.83,117.79,107.79,108.76
BEGIN DESCRIPTION:
Upstream Section - QUEENSTON BLVD
END DESCRIPTION:
Node Name=P
XS GIS Cut Line= 6
3023882.0114718713879647.20052093023921.3716293613878899.3699956
3023930.6491698613878700.71192843023937.6672004513878476.5017468
3023947.4394906213878357.06432173024029.95999487 13877915.145258
#Sta/Elev= 30
       0  121.86  366.02  121.98  658.45     121  679.14  117.99  694.08  117.64
  748.87   117.9  783.67  119.53  813.88  117.01  830.49  112.04   893.4  103.83
  917.48   104.2  919.68  101.96  936.87  100.62  941.76   98.18  948.25  100.69
   950.8     104  957.48  103.98  975.58  109.06  995.47  117.58 1008.86  119.89
 1067.87  120.42 1087.72  119.58 1187.05  119.72  1296.9  118.34 1341.86  119.16
 1411.79  118.68 1491.71  119.53 1616.58  119.03 1666.54  120.09 1741.46  119.78
#Mann= 4 ,-1 , 0
       0     .15       0  658.45     .07       0  783.67     .04       0
 1008.86     .07       0
#XS Ineff= 2 ,-1
       0  833.39  118.77 1008.85 1741.46  118.81
Permanent Ineff=
       F       F
#Block Obstruct= 2 , 0
       0                 1636.57       0  119.87
Bank Sta=783.67,1008.86
XS Rating Curve= 0 ,0
Exp/Cntr=0.5,0.3

Type RM Length L Ch R = 3 ,66899.86,,,
BEGIN DESCRIPTION:
QUEENSTON BLVD
END DESCRIPTION:
Node Name=QUEENSTON BLVD
Bridge Culvert--1,0,-1,-1, 0
Deck Dist Width WeirC Skew NumUp NumDn MinLoCord MaxHiCord MaxSubmerge Is_Ogee
9.5,90,2.6,0, 60, 60, , , 0.98, 0, 0,0,,
       0   84.09  103.87  118.71  168.17   192.9  222.58  232.47   257.2  262.15
   267.1  291.83  351.18   484.9  514.78  559.61  614.39  624.35  654.24  669.18
   738.9  748.87  763.78  768.75   778.7  803.56   813.5  818.47  828.42  833.39
 1008.85 1013.56 1028.18 1033.14  1038.1 1057.95 1062.91 1072.83 1092.68  1142.3
 1157.18 1167.11 1172.07 1197.03 1217.01 1346.85 1366.83 1411.79  1496.7 1546.65
 1571.63  1601.6 1616.58 1626.57 1636.56 1661.54 1691.51 1721.48 1736.47 1741.46
  120.36  120.27  119.95  120.36  120.62  121.03  121.16  121.01  121.15  121.34
  121.14  121.37  121.15  121.71  121.54  121.87  121.68  121.46  122.03  121.75
  121.69  121.38  121.23  121.11  120.24  119.57  118.77  125.25  125.49  125.55
  125.85   125.8  125.53  121.71   121.8  121.51  121.74   121.2  120.73  120.32
   119.5  119.35  119.48   119.2  119.59   118.8  119.08  118.95  119.65  119.52
  119.81  119.85   120.1  119.96  120.16  119.37  119.41  120.38  120.47  120.29
       0       0       0       0       0       0       0       0       0       0
       0       0       0       0       0       0       0       0       0       0
       0       0       0       0       0       0       0       0       0  119.74
  120.04       0       0       0       0       0       0       0       0       0
       0       0       0       0       0       0       0       0       0       0
       0       0       0       0       0       0       0       0       0       0
       0   84.09  103.87  118.71  168.17   192.9  222.58  232.47   257.2  262.15
   267.1  291.83  351.18   484.9  514.78  559.61  614.39  624.35  654.24  669.18
   738.9  748.87  763.78  768.75   778.7  803.56   813.5  818.47  828.42  833.39
 1008.85 1013.56 1028.18 1033.14  1038.1 1057.95 1062.91 1072.83 1092.68  1142.3
 1157.18 1167.11 1172.07 1197.03 1217.01 1346.85 1366.83 1411.79  1496.7 1546.65
 1571.63  1601.6 1616.58 1626.57 1636.56 1661.54 1691.51 1721.48 1736.47 1741.46
  120.36  120.27  119.95  120.36  120.62  121.03  121.16  121.01  121.15  121.34
  121.14  121.37  121.15  121.71  121.54  121.87  121.68  121.46  122.03  121.75
  121.69  121.38  121.23  121.11  120.24  119.57  118.77  125.25  125.49  125.55
  125.85   125.8  125.53  121.71   121.8  121.51  121.74   121.2  120.73  120.32
   119.5  119.35  119.48   119.2  119.59   118.8  119.08  118.95  119.65  119.52
  119.81  119.85   120.1  119.96  120.16  119.37  119.41  120.38  120.47  120.29
       0       0       0       0       0       0       0       0       0       0
       0       0       0       0       0       0       0       0       0       0
       0       0       0       0       0       0       0       0       0  119.64
  119.94       0       0       0       0       0       0       0       0       0
       0       0       0       0       0       0       0       0       0       0
       0       0       0       0       0       0       0       0       0       0
Pier Skew, UpSta & Num, DnSta & Num=  ,888.56, 2 ,888.56, 2 , 0 , 0 , 0 ,,
     1.4     1.4
      95     121
     1.4     1.4
      95     121
Pier Skew, UpSta & Num, DnSta & Num=  ,944.46, 2 ,944.46, 2 , 0 , 0 , 0 ,,
     1.4     1.4
      95     121
     1.4     1.4
      95     121
Abutment Skew #Up #Dn= , 2 , 2
  830.66  900.96
  119.74  103.49
  830.66  900.96
  119.64  103.39
Abutment Skew #Up #Dn= , 2 , 2
  965.16 1011.15
  103.97  120.04
  965.16 1011.15
  103.87  119.94
BR Coef=-1 , 1 , 1 ,0.9, 0 ,,,0.8,-1,1.2,0,
WSPro=,,,, 1 ,,,, 0 ,,,, 0 ,,,,-1 ,-1 ,-1 , 0 , 0 , 0 , 0 , 0
BC Design=,, 0 ,, 0 ,,,,,,
BC Use User HTab Curves=0
BC User HTab FreeFlow(D)= 0

Type RM Length L Ch R = 1 ,66850.04,184,184.36,178.27
BEGIN DESCRIPTION:
Downstream Section - QUEENSTON BLVD
END DESCRIPTION:
XS GIS Cut Line= 6
 3023987.973202213879648.85701373024027.3333596913878901.0264883
3024036.6109001913878702.36842113024043.6289307813878478.1582396
3024053.4012209513878358.7208144 3024135.921725213877916.8017508
#Sta/Elev= 30
       0  120.57  474.94  120.21  783.67  117.91   813.5  118.42  828.42   119.8
  833.39  119.03  868.19   106.3  883.11  104.28  902.99  105.67  907.97   104.8
  917.91  101.27  926.94  100.01  957.14  103.14  971.25   105.8  980.65  105.56
  990.05  106.58 1028.18  120.44  1038.1  121.11 1067.87   121.1 1082.76   120.2
 1092.68  120.69 1162.14  119.03 1301.89  118.05 1381.82  119.24 1411.79  118.58
 1461.74  119.26 1526.67  118.96 1556.64  119.93 1586.61  119.44 1741.46  119.83
#Mann= 3 ,-1 , 0
       0     .07       0  828.42     .04       0  1038.1     .07       0
#XS Ineff= 2 ,-1
       0  833.39  118.77 1008.85 1741.46  118.81
Permanent Ineff=
       F       F
#Block Obstruct= 2 , 0
       0                 1556.64       0  119.93
Bank Sta=828.42,1038.1
XS Rating Curve= 0 ,0
Exp/Cntr=0.5,0.3

Type RM Length L Ch R = 1 ,66665.68,564.89,547.93,507.48
XS GIS Cut Line= 4
3024215.1617241913879650.96790193024215.1617241913879168.0958361
3024215.16172419 13878548.5376923024207.87269677 13877928.979876
#Sta/Elev= 30
       0  119.47  393.27  120.18  512.85  119.75  607.78  118.19  697.72  118.08
  732.69  118.95  792.65  117.59  822.63  118.31  832.62   117.2  857.61   108.5
  872.59  104.78  887.58  103.36  917.56  104.75  930.44  101.21  940.15   99.84
  950.96  100.96  962.53  104.38  977.52  106.67  1012.5  118.13 1022.49  119.46
 1042.47  118.43 1057.46  119.98 1072.45   120.3  1157.4  118.99 1187.38  120.17
 1242.34  120.08  1297.3  118.39 1392.24  118.06 1532.15  120.35 1722.03  119.72
#Mann= 3 ,-1 , 0
       0     .07       0  822.63     .04       0 1022.49     .07       0
#XS Ineff= 2 ,-1
       0  672.74  118.59 1277.32 1722.03  118.95
Permanent Ineff=
       F       F
#Block Obstruct= 2 , 0
       0   94.58  120.23               0
Bank Sta=822.63,1022.49
XS Rating Curve= 0 ,0
Exp/Cntr=0.3,0.1

Type RM Length L Ch R = 1 ,66117.75,192.48,206.18,221.1
Node Name=O
XS GIS Cut Line= 5
3024916.7370926913879128.22813373024869.0199965213879002.3300915
3024737.89985195 13878656.3799963024601.4001249413878302.7301128
3024468.8564267813877946.1068103
#Sta/Elev= 30
       0  119.29  159.64  118.64  249.63  116.02  339.62  115.86  384.61  118.91
  399.83  117.45  409.61  116.63  424.61  117.42  439.61  115.27   474.6  105.39
   489.6   99.32   494.6   99.01  514.58  100.19  529.54  104.38   544.5  104.15
  554.48  105.24  574.43  109.86  599.37  117.86  609.35  118.99  649.25  116.27
  662.93  117.04  749.01  118.24  773.95  116.99  853.75  116.47  878.69  117.58
  942.97  116.87 1002.26  119.12 1026.97   118.2 1142.38  119.17 1264.14     120
#Mann= 6 ,-1 , 0
       0     .15       0  399.83     .07       0  424.61     .04       0
  609.35     .07       0  662.93     .15       0 1142.38     .07       0
#XS Ineff= 1 ,-1
       0  354.62   116.9
Permanent Ineff=
       F
Bank Sta=424.61,609.35
XS Rating Curve= 0 ,0
Exp/Cntr=0.3,0.1

Type RM Length L Ch R = 1 ,65911.57,683.48,718.37,692
XS GIS Cut Line= 5
3025087.9562384513879258.05333343025016.9426009513878971.2950486
3024918.86996244 13878575.2699223024812.8527860313877856.0905861
3024546.5485286113877138.7652491
#Sta/Elev= 30
       0  117.92  108.32  118.54  211.72  115.86   320.3  119.35  355.13  118.91
   399.9  115.81  439.71  115.77  544.19  120.27  600.71  118.03  613.85  115.76
  633.75   117.3   643.7  115.91  678.53  105.79   728.3   99.16  758.18   104.7
  793.03  116.23  807.97  119.35  852.11   117.3  862.74   119.4  947.39  119.51
 1046.97  117.18 1315.84   120.9  1455.2   119.6 1554.57  120.35 1683.76  117.44
 1808.41  119.96 2066.34  120.36 2145.83  120.04 2160.74  118.82 2195.52  120.45
#Mann= 6 ,-1 , 0
       0     .15       0  600.71     .07       0  633.75     .04       0
  807.97     .07       0  852.11     .15       0 1808.41     .07       0
#XS Ineff= 2 ,-1
       0  474.54  116.89 1648.98 2195.52  118.65
Permanent Ineff=
       F       F
#Block Obstruct= 2 , 0
       0   34.47  118.75               0
Bank Sta=633.75,807.97
XS Rating Curve= 0 ,0
Exp/Cntr=0.3,0.1

Type RM Length L Ch R = 1 ,65193.2 ,580.49,620.8,606.15
XS GIS Cut Line= 6
3025609.9699581913879312.22940613025578.18918186 13879073.339792
3025548.0301214513878846.64011423025525.2998519413878619.3698994
3025468.8554110213877841.51285943025372.9579650313877156.8383757
#Sta/Elev= 30
       0   119.4  191.81  117.78  245.97  115.21  270.82  115.16  315.57  117.96
  385.17  118.19     415  117.17  434.89  115.98  464.72  106.12  496.08    98.5
  503.71   98.98  509.41  102.15  519.34  103.93  539.21  103.41  559.07   105.5
  598.79  117.19  608.72  118.19  643.48  117.05  671.08  118.98  793.08  118.05
  858.08  116.09 1053.05  118.99 1378.01  117.84    1408  119.12    1458  119.16
 1482.97  117.88 1642.13  116.82 1808.87  119.76 2104.69  119.51 2169.35  120.86
#Mann= 6 ,-1 , 0
       0     .15       0  385.17     .07       0     415     .04       0
  608.72     .07       0  671.08     .15       0 1808.87     .07       0
#XS Ineff= 2 ,-1
       0  285.74  116.33 1477.99 2169.35  118.17
Permanent Ineff=
       F       F
Bank Sta=415,608.72
XS Rating Curve= 0 ,0
Exp/Cntr=0.3,0.1

Type RM Length L Ch R = 1 ,64572.4 ,535.53,513.87,510.91
Node Name=N
XS GIS Cut Line= 5
3026013.6850300313879276.8187158 3026015.524265213879153.5177813
3026025.29983619  13878498.159843026022.8132926113877819.6461052
3026008.8077431913877168.0617784
#Sta/Elev= 30
       0  117.64  103.58  117.43   182.9  114.74  262.35  117.51  376.55  117.91
   441.1  114.71  505.65  117.11  592.54  117.71  629.78  118.01  659.58  116.31
  669.51  117.37  689.37  115.17  729.09  103.39  743.99  102.89  763.85  105.74
  778.75  103.25  788.72   98.41  799.56   97.94  813.67    98.3  818.66     100
  838.61  112.66  853.58  115.95  888.51  114.15  903.47  116.11  923.43  115.11
 1098.05  117.32 1462.24  116.52  2009.5  118.77 2074.17  117.48    2109  119.03
#Mann= 4 ,-1 , 0
       0     .15       0  592.54     .07       0  669.51     .04       0
  853.58     .07       0
#XS Ineff= 1 ,-1
       0  470.89  115.29
Permanent Ineff=
       F
Bank Sta=669.51,853.58
XS Rating Curve= 0 ,0
Exp/Cntr=0.3,0.1

Type RM Length L Ch R = 1 ,64058.53,540.56,519.63,518.22
Node Name=M
XS GIS Cut Line= 5
3026482.0151301213879197.25128963026529.9799291913878767.3000498
 3026536.820138613878370.93995013026518.4596110313877921.6908486
3026486.2746360313877134.1786441
#Sta/Elev= 30
       0  116.86  159.12  116.41  273.49  113.65  348.08  116.13  426.12  116.04
  442.53  114.78  467.31  115.69   472.5  115.52  498.38  107.48  612.45  105.28
  638.41   99.99   664.5  100.67  667.46   97.68  672.77   97.47  680.17   97.68
  683.24  100.54   702.4    99.9  759.66  114.13  769.57  115.29  799.31  114.29
  854.02  116.75  923.96  115.84 1268.67  116.96 1288.64  118.82 1373.44  120.31
  1737.6  119.93 1977.04  118.16 2006.97  119.15 2046.88  117.96 2066.83  118.81
#Mann= 4 ,-1 , 0
       0     .15       0  426.12     .07       0  467.31     .04       0
  769.57     .07       0
#XS Ineff= 1 ,-1
       0  318.25  115.13
Permanent Ineff=
       F
Bank Sta=467.31,769.57
XS Rating Curve= 0 ,0
Exp/Cntr=0.3,0.1

Type RM Length L Ch R = 1 ,63538.9 ,379,377.01,377.92
XS GIS Cut Line= 4
 3026999.528202713879787.65365213027053.1301296113878555.8001447
3027057.83943778 13877666.5788263027059.9316251913877271.5563221
#Sta/Elev= 30
       0  116.73   29.95  117.17   79.87  114.91  109.82  114.83  164.74  117.36
  419.33  117.83  668.93  117.26  851.79  115.17  943.48  113.16 1108.22  114.27
 1128.19  114.15 1143.16  112.72 1158.14  113.77 1168.12  112.53 1203.07   102.4
 1213.05  100.87 1228.03  101.23 1238.02   98.33 1247.97    97.3    1258   97.84
 1287.97  102.83 1332.93  113.51 1347.92  114.49 1447.84  113.19 2137.07  118.77
 2334.59  118.89 2423.47  116.75 2472.85  118.12 2502.47  116.85 2517.29  118.32
#Mann= 4 ,-1 , 0
       0     .15       0  851.79     .07       0 1158.14     .04       0
 1347.92     .07       0
#Block Obstruct= 2 , 0
       0  164.74     116               0
Bank Sta=1158.14,1347.92
XS Rating Curve= 0 ,0
Exp/Cntr=0.3,0.1

Type RM Length L Ch R = 1 ,63161.89,201.27,215.62,212.55
Node Name=L
XS GIS Cut Line= 5
3027202.9835044413879928.37843633027210.9067169413879700.1866354
 3027222.856496213879356.03345233027426.2642258613878829.9239403
3027443.1890607813877538.8481103
#Sta/Elev= 30
       0  116.82  707.47   116.2  717.45  113.02  742.41   99.65   747.4   98.86
  762.38   101.8  782.34  101.18  797.32  104.12  812.29  104.25  852.23  114.01
  892.16  112.59 1011.96  115.27 1071.86  116.83 1101.81  119.92 1321.21  114.59
 1331.18  113.82 1376.05  100.64 1400.97  101.37 1421.51   97.18 1445.84  101.41
 1465.78  100.96 1510.65  114.39 1520.62  115.28  1630.3  117.23 1655.22  115.58
 1779.86  115.67 1974.28  118.12 2168.71  117.72 2223.55  115.84 2427.95  118.26
#Mann= 3 ,-1 , 0
       0     .07       0 1321.21     .04       0 1520.62     .07       0
#XS Ineff= 1 ,-1
  702.47  912.13  114.07
Permanent Ineff=
       T
Bank Sta=1321.21,1520.62
XS Rating Curve= 0 ,0
Exp/Cntr=0.3,0.1

Type RM Length L Ch R = 1 ,62946.27,809.47,883.26,888.34
Node Name=K
XS GIS Cut Line= 6
 3027814.463252613880481.25856413027769.73991686 13879443.779996
3027715.2200127813879303.56997463027590.1021527813879043.0494983
3027637.3300766913878571.37983793027707.4300021113877379.6200823
#Sta/Elev= 30
       0  116.78  216.93  116.44  713.66  114.37  883.55     119  938.51  118.64
  963.49  115.29  973.49  117.76 1048.15   114.6 1243.69   115.9 1258.64  114.26
 1288.54   99.95  1298.5   98.42 1318.43   98.92  1328.4  104.02 1363.28  106.43
 1393.18  113.47 1447.99  115.37  1472.9  113.24 1642.55  117.25  1862.1   115.3
 1926.97   99.79 1976.89  103.83 2001.76   97.11 2011.86   98.03 2061.81  115.06
 2081.79   115.9 2706.17  116.75 2761.11  114.98 2866.01  117.42 3145.73  117.98
#Mann= 4 ,-1 , 0
       0      .1       0  216.93     .07       0  1862.1     .04       0
 2081.79     .07       0
#XS Ineff= 2 ,-1
 1258.64 1393.18  113.47 2806.07 3145.73  116.64
Permanent Ineff=
       T       F
Bank Sta=1862.1,2081.79
XS Rating Curve= 0 ,0
Exp/Cntr=0.3,0.1

Type RM Length L Ch R = 1 ,62063.01,376.66,291.66,178.64
XS GIS Cut Line= 5
 3027986.516386213880540.36868213028015.3299768613880400.5100379
3028282.8199274413879102.13993133028433.1598498713878832.2198674
3028468.3677846913877443.4486949
#Sta/Elev= 30
       0  115.97   225.9  114.31 1024.89  114.34 1094.66   113.7 1109.61  109.32
 1159.45  106.21 1189.35  112.91 1279.06  113.27 1294.01   112.7 1333.88  103.01
 1368.76  102.72 1398.66  103.16 1438.53     111 1493.35  111.34 1502.46  111.12
  1545.9    98.2 1591.35   96.83 1599.86   99.74 1654.54   98.76 1707.63  113.83
  1782.4  115.93 1982.28  112.11 2347.08  114.45 2547.44  112.43 2581.95  116.02
  2661.9  115.84 2711.87  112.55 2866.79  116.74  3021.7  113.68 3166.62  117.85
#Mann= 5 ,-1 , 0
       0      .1       0   225.9     .07       0 1493.35     .04       0
 1707.63     .07       0 2547.44     .15       0
#XS Ineff= 2 ,-1
       0  735.84  114.52 2392.05 3166.62  114.46
Permanent Ineff=
       F       F
#Block Obstruct= 2 ,-1
 1094.36  1204.3  113.04 1298.99 1438.53   110.5
Bank Sta=1493.35,1707.63
XS Rating Curve= 0 ,0
Exp/Cntr=0.3,0.1

Type RM Length L Ch R = 1 ,61771.35,482.51,533.88,531.47
XS GIS Cut Line= 6
 3029116.770031213880423.6723932 3029037.831212713880190.0130836
 3028666.046523213879089.5303764 3028554.5113132 13878873.895309
 3028456.503635213878728.97204243028493.33492637 13877457.319402
#Sta/Elev= 30
       0  117.56  590.62  113.85  605.58  109.88  635.49  106.43   665.4  109.64
  680.36  113.53  705.29  112.33  740.18  114.55  924.64  115.16 1418.13   111.7
 1472.63  100.84 1521.58   96.61 1526.87   97.09 1532.08  100.42 1576.67  100.06
  1606.4  102.34 1655.99  112.64 1725.97  112.22 1770.96  107.39 1825.94  113.33
 2314.87  114.12  2389.7  111.68 2485.94  112.01 2519.42  115.52 2609.22  115.73
 2674.08  112.44 2713.99  115.65 2808.78  116.96 2933.51  113.48 3098.14  117.97
#Mann= 4 ,-1 , 0
       0     .07       0 1418.13     .04       0 1655.99     .07       0
 2485.94     .15       0
#XS Ineff= 2 ,-1
       0  924.64  115.16 2314.87 3098.14  114.12
Permanent Ineff=
       F       F
#Block Obstruct= 1 ,-1
  590.62  680.36  113.03
Bank Sta=1418.13,1655.99
XS Rating Curve= 0 ,0
Exp/Cntr=0.3,0.1

Type RM Length L Ch R = 1 ,61237.47,624.28,656.92,600.63
XS GIS Cut Line= 4
3029447.7454191113880079.36041783029031.0999269513878808.2999678
3028969.60004994 13878511.0298933028980.2532438613877505.3307889
#Sta/Elev= 30
       0  119.03   99.82  118.16  139.75  116.69  159.71  113.64  174.69   115.6
  189.66  114.33  209.62  114.73  234.58   108.7  259.54  107.25  299.46  114.03
  339.39  113.88  349.37  115.11  404.28  113.03 1287.69  111.68  1337.6  110.52
 1372.44  111.79 1378.36   111.5 1437.47   97.73 1490.39   98.12 1492.94    96.2
 1511.52   98.23 1533.99   97.93 1577.73   110.9  1591.4  111.77 1889.33  111.44
 2019.39  111.78  2071.6  112.55 2256.34  113.66 2442.79  112.56 2646.93  115.99
#Mann= 7 ,-1 , 0
       0     .07       0 1372.44     .04       0  1591.4     .12       0
 1889.33     .07       0 2019.39     .15       0  2071.6     .07       0
 2256.34     .15       0
#XS Ineff= 2 ,-1
       0  349.37  115.11 1974.76 2646.93  112.49
Permanent Ineff=
       F       F
#Block Obstruct= 1 ,-1
  209.62   299.4   113.5
Bank Sta=1372.44,1591.4
XS Rating Curve= 0 ,0
Exp/Cntr=0.3,0.1

Type RM Length L Ch R = 1 ,60580.55,550.11,551.19,554.75
XS GIS Cut Line= 4
3030010.1301211113880051.18002793029608.6099267813878740.5799589
3029305.7122386113877894.55277953028997.6144296113877359.4974192
#Sta/Elev= 30
       0  117.19   66.39  116.79  214.33  118.45  348.91  115.45  742.68  114.07
 1036.77   110.6 1086.61  112.11 1236.15  111.25 1276.02  108.58  1315.9   98.61
 1352.76   95.79 1420.65   98.49 1490.54  111.24 1535.48  108.89 1681.93  112.08
 1861.68  110.66 2009.75  110.08 2074.65  112.79 2134.55  111.66 2258.85  113.62
  2329.1  113.96 2358.97  111.48 2403.79  111.49 2458.56  114.85    2593  114.79
  2687.6  112.57 2822.04  115.25    2832  117.23 2841.96  115.55 2886.77  116.49
#Mann= 7 ,-1 , 0
       0     .12       0   66.39     .07       0 1236.15     .04       0
 1490.54     .07       0 1681.93     .12       0 1861.68     .07       0
 2258.85     .15       0
#XS Ineff= 1 ,-1
 1681.93 2886.77  112.11
Permanent Ineff=
       F
Bank Sta=1236.15,1490.54
XS Rating Curve= 0 ,0
Exp/Cntr=0.3,0.1

Type RM Length L Ch R = 1 ,60029.36,485.91,497.69,507.81
XS GIS Cut Line= 5
3030667.8207348613880016.25293243030168.9099872713878695.5400227
3030073.2399030313878391.43990913029422.9616760313877448.0392369
3029008.0310754513877248.3864209
#Sta/Elev= 30
       0  117.44  261.31   116.5  728.35  113.11 1406.82  111.27 1426.75  107.17
 1454.48  107.93 1490.27   97.93 1540.95   97.76 1558.82   95.45 1571.83   95.61
 1578.17   97.55 1594.61      98  1650.9  112.31 1765.47  113.56 1919.91   110.5
 1974.71  111.83 2009.58  110.32 2367.51  113.17 2512.73  110.96 2572.52  112.57
    2712  113.15 2796.69  112.23  2821.6  114.64 2851.49  115.18 2911.06  114.31
 2935.82  112.27 2960.57  112.02 2990.28  114.32 3173.48  114.63 3336.87  116.37
#Mann= 5 ,-1 , 0
       0     .12       0  261.31     .07       0 1406.82     .04       0
  1650.9     .07       0 2367.51     .15       0
#XS Ineff= 1 ,-1
 1954.78 3336.87  112.05
Permanent Ineff=
       F
Bank Sta=1406.82,1650.9
XS Rating Curve= 0 ,0
Exp/Cntr=0.3,0.1

Type RM Length L Ch R = 1 ,59531.67,90.71,100.56,109.04
XS GIS Cut Line= 5
3030803.0425772813880098.32429063030630.0875426113878567.3535993
3030569.2333336213878256.67541483029731.0827789513877103.6869072
3029024.1583397813876718.5078875
#Sta/Elev= 30
       0   118.7   64.82  116.47  316.11  116.36 1560.49  111.19 1605.01  109.32
 1643.13   97.98  1694.8   98.76 1699.51    95.7 1712.47   95.85 1716.32   99.22
 1754.34   98.22 1792.98  109.87 1807.82  111.79 1961.96  110.14 2076.59  111.62
 2151.35  108.81 2373.32  111.14 2714.55  111.47 2839.15  108.84  2948.8  112.89
  3073.4  109.65 3108.29  111.94 3252.83  112.11 3282.73  117.08  3580.9  116.96
 3650.47  114.36 3700.16  116.49 3814.46  116.46 3933.73  113.74 4087.78  116.83
#Mann= 5 ,-1 , 0
       0     .12       0  316.11     .07       0 1560.49     .04       0
 1807.82     .07       0 2373.32     .15       0
#XS Ineff= 1 ,-1
 1907.13 4087.78  112.15
Permanent Ineff=
       F
Bank Sta=1560.49,1807.82
XS Rating Curve= 0 ,0
Exp/Cntr=0.3,0.1

Type RM Length L Ch R = 1 ,59431.11,152,128.09,109.1
Node Name=J
XS GIS Cut Line= 6
3030849.4840854413880104.1963261 3030690.219640213878306.8820073
 3030641.883122713878296.45650333030589.7556022713878257.5976571
 3029752.501043213877091.92971283029236.8321270213876568.3343033
#Sta/Elev= 30
       0  118.64  317.74  116.86   549.8  114.28 1574.44  111.19 1599.43  108.58
 1624.42  108.87 1660.46   97.53 1710.68   97.49 1721.32    95.3 1727.68    95.3
  1731.9   99.41 1770.57   98.23 1804.36  111.23 2103.21  111.67 2182.94  108.69
 2431.95  110.85 2785.92  111.66 2900.53  108.91 3025.12  113.01 3129.77  109.82
 3259.33  112.92  3329.1  111.82 3359.02   117.1    3489  117.19 3538.99  114.47
 3723.96  116.73 3803.95  113.78 3948.93  117.38 3968.92  115.75  4088.9  116.26
#Mann= 5 ,-1 , 0
       0     .12       0  317.74     .07       0 1574.44     .04       0
 1804.36     .07       0 2431.95     .15       0
#XS Ineff= 1 ,-1
 1958.69  4088.9  112.37
Permanent Ineff=
       F
Bank Sta=1574.44,1804.36
XS Rating Curve= 0 ,0
Exp/Cntr=0.3,0.1

Type RM Length L Ch R = 1 ,59303.02,227.93,132.65,34.23
XS GIS Cut Line= 6
3031340.5903866913879903.48314483030879.37739836 13878532.655834
3030796.5383251913878301.61955073030647.4073898613878285.1714209
3030614.5108021113878255.56452473029328.9457879413876477.9253634
#Sta/Elev= 30
       0  119.47  100.47  118.08  1485.6   111.1 1500.33  109.29 1524.92  110.23
 1558.39   97.71 1597.07   97.57 1606.98   95.26  1615.5   96.01 1619.52  100.16
 1660.18   97.72  1683.1  109.31 1696.56   111.2 1926.23  112.56  1986.2  110.55
 2111.13  111.08 2151.11  108.78 2396.12  110.72 2770.77  111.37 2880.72  108.99
 3005.65  112.94 3135.58  109.76 3240.52  113.05 3310.48  111.78 3340.47  117.24
 3495.39  114.29 3605.33  116.33 3790.23  114.56  3840.2  117.03 4080.07  115.54
#Mann= 5 ,-1 , 0
       0      .1       0  100.47     .07       0  1485.6     .04       0
 1696.56     .07       0 2396.12     .15       0
#XS Ineff= 1 ,-1
 1926.23 4080.07  112.56
Permanent Ineff=
       F
Bank Sta=1485.6,1696.56
XS Rating Curve= 0 ,0
Exp/Cntr=0.5,0.3
